HEC-RAS study Baxter.prj: Baxter River GIS Example

--- Baxter.g02 (geometry) --- (continued)

Type RM Length L Ch R = 1 ,58425.  ,441.7,403.69,386.57
XS GIS Cut Line= 4
 6430885.8606241 2048342.2654694 6431107.8318126 2048799.6605337
 6431107.8318126 2049270.5084276 6431471.0573077  2050192.025042
#Sta/Elev= 30
       0   95.84  180.18   95.84  209.07    93.4  281.95   81.84  336.27   71.84
  358.34   65.84  419.35   63.32  662.45   55.84  728.69   49.84  748.38   45.84
  754.36   41.64  772.99   30.95  799.19      32  816.85   28.44  821.98   30.08
  837.09   27.88  862.08      32  887.22      40  893.23   45.84  904.94   49.54
   921.8   55.84 1070.59   55.84 1078.01   57.84 1169.13   63.84 1283.51   69.84
 1466.82   71.99 1497.26   73.84 1519.44   83.84 1643.57   85.84 1969.78   85.84
#Mann= 2 ,-1 , 0
       0     .06       0  419.35    .035       0
Bank Sta=754.36,904.94
XS Rating Curve= 0 ,0
Exp/Cntr=0.3,0.1

Type RM Length L Ch R = 1 ,58021.  ,581.56,561.67,525.46
XS GIS Cut Line= 5
 6430569.7199136 2048422.9822092 6430647.1710139 2048632.2932755
 6430735.1786535 2049365.6900038 6430999.2014303 2050084.4187843
 6431128.0109857 2050333.2794433
#Sta/Elev= 30
       0   95.37  286.88   93.84  328.65   89.38  384.76   79.08  465.98   63.84
  604.81   55.84  613.37   53.84  623.11   45.84  639.46   42.59  652.59      40
  663.92   39.88  678.75   32.54  712.84   31.88  721.37   29.88  726.76   31.64
   742.6   30.68  760.29      32  782.19   45.84  805.81    50.3  840.43   55.84
 1094.79   55.84 1186.69   63.84 1272.21   67.84 1560.37   71.84 1608.86   73.84
 1621.76   75.84 1640.04   83.84 1648.53   85.84 1839.01   87.15 2007.75   86.19
#Mann= 2 ,-1 , 0
       0     .06       0  384.76    .035       0
Bank Sta=639.46,805.81
XS Rating Curve= 0 ,0
Exp/Cntr=0.3,0.1

Type RM Length L Ch R = 1 ,57459.  ,448.27,460.04,476.86
XS GIS Cut Line= 3
 6430031.6080147 2048685.3117913 6430193.0415891 2049371.4044352
 6430690.7950945 2050575.4297576
#Sta/Elev= 30
       0   91.84   42.61   91.84  117.75   87.84  219.53   86.41  253.81   85.84
  385.87    57.8   401.8   53.84  414.88   45.84  437.24      40  447.55    41.5
  463.86   34.75  563.85   32.75  595.38   39.05   609.7   45.84  651.05   53.84
  671.21   59.84  722.72   55.89  765.75   57.84  813.51   57.84  866.43   55.84
  902.41   57.27  918.85   55.84  972.33   55.84  1099.1   68.44 1199.57    72.6
 1275.18   72.13  1430.5   75.84 1537.21   85.84 1735.71   87.84 2007.69   87.84
#Mann= 2 ,-1 , 0
       0     .06       0  219.53    .035       0
Bank Sta=385.87,595.38
XS Rating Curve= 0 ,0
Exp/Cntr=0.3,0.1

Type RM Length L Ch R = 1 ,56999.  ,356.17,351.22,350.04
XS GIS Cut Line= 3
  6429574.212903   2048544.05739 6429722.1936953 2049418.4892199
 6430152.6831955 2051012.6456962
#Sta/Elev= 30
       0   92.16  117.73   89.84  130.22   87.84  440.07   86.62  522.27   85.23
  527.97   83.84  560.63   63.84  582.94   56.32  606.77   45.84   637.4    41.1
  656.14    41.5   678.8      36  733.24   35.05   741.4   33.57  752.17    35.5
  785.16      33  802.36      40  808.48   45.84  822.89   49.31  866.74   59.84
  962.29   59.84 1105.69   55.84 1167.87   55.84 1308.92   69.84 1353.67   81.84
 1689.62   84.48 2108.58   81.84 2147.78   87.84 2257.19   89.84 2538.12   89.84
#Mann= 2 ,-1 , 0
       0     .06       0  440.07    .035       0
Bank Sta=582.94,822.89
XS Rating Curve= 0 ,0
Exp/Cntr=0.3,0.1

Type RM Length L Ch R = 1 ,56648.  ,522.44,542.07,563.75
XS GIS Cut Line= 3
 6429184.0817964 2048476.7934323 6429385.8737644 2049505.9323981
 6429782.7312621 2050965.5609115
#Sta/Elev= 30
       0   89.99   125.1   87.84  134.44   85.84  576.06   85.84  627.48   85.84
  675.12   77.84  687.12   73.84  712.53   53.84  718.93      52  735.79   47.84
  800.15   45.84  806.04   41.87  814.84    41.5  823.13      37  891.33   36.36
  918.78   33.48  950.85      40  961.44   53.84  964.46   54.76  987.51   59.84
 1092.56   59.84 1253.54   53.84 1310.42   53.84 1374.04   63.84 1543.04   71.84
 1619.37   83.84 1951.18   86.98 2410.53   85.84 2442.68   89.84 2561.35   91.44
#Mann= 2 ,-1 , 0
       0     .06       0  576.06    .035       0
Bank Sta=718.93,964.46
XS Rating Curve= 0 ,0
Exp/Cntr=0.3,0.1

Type RM Length L Ch R = 1 ,56106.  ,617.86,622.85,632.88
XS GIS Cut Line= 4
 6428694.3159041 2048460.8182062 6428799.0112454 2049233.6785681
  6428828.347141  2049571.041084  6429051.655807 2050899.1377053
#Sta/Elev= 30
       0   87.07  618.97   85.84  680.03   78.45  692.74   73.84  763.45   63.84
  791.55   53.84  804.58   50.96  853.73      42   863.3    38.4  978.63    37.1
  997.44    34.4 1020.76    40.1 1029.79   45.84 1038.03   53.87 1073.71   61.84
 1104.26   61.84 1195.37   57.84 1387.46   53.84 1415.45   63.84 1447.15   67.84
 1472.72   73.84  1489.3   73.84 1507.49   69.84 1646.03   71.84 1667.86   75.84
 1737.95   75.84 1746.94   78.67 1793.12   85.84 1878.53   90.06 2465.29   90.39
#Mann= 2 ,-1 , 0
       0     .06       0  680.03    .035       0
Bank Sta=804.58,1038.03
XS Rating Curve= 0 ,0
Exp/Cntr=0.3,0.1

Type RM Length L Ch R = 1 ,55483.  ,407.38,425.15,445.81
XS GIS Cut Line= 4
 6428185.6320133 2048509.1642128 6428177.2240245 2049265.8840574
  6428202.447991 2049551.7560081 6428261.3040073 2051023.1556585
#Sta/Elev= 30
       0   87.27  494.97   85.84  529.07   81.84  560.01   73.84  598.71   68.49
  738.65   65.84  799.25   50.23  808.22   45.84  862.81   36.71  921.46    35.2
  939.41      37  970.78    34.6 1028.01   45.84  1045.2   55.84 1069.46   59.08
  1184.1   58.67 1249.41   57.84 1276.65   51.84 1308.76   53.84 1361.57   51.84
 1400.79   63.84 1439.62   67.84 1476.34   77.84 1493.15   77.84 1507.18   73.84
 1582.19   75.83 1613.99   83.84 1666.29   87.91 2249.73   93.84 2516.33   93.84
#Mann= 2 ,-1 , 0
       0     .06       0  598.71    .035       0
Bank Sta=799.25,1045.2
XS Rating Curve= 0 ,0
Exp/Cntr=0.3,0.1

Type RM Length L Ch R = 1 ,55058.  ,629.67,685.71,707.67
XS GIS Cut Line= 4
 6427706.3761307 2048376.7382235 6427772.2558447 2049116.3351276
 6427757.5878969 2049952.4073959 6427769.4360941 2050857.0977139
#Sta/Elev= 30
       0   91.05  531.51   85.84  577.05   81.84  644.92   69.98  687.67   67.84
  912.63   65.84  931.52      59  964.66   47.86 1017.19   36.52 1074.43   35.12
 1101.38      37 1132.86    34.6 1161.01    38.5 1190.01   45.84 1197.86   53.84
 1201.91   55.13 1310.51   58.38 1419.55   57.84 1423.46   51.84 1431.69   53.84
 1440.35   51.84 1471.48   51.84  1518.3   65.84 1544.11   69.84 1715.57   75.84
 1723.74   77.84 1761.21   77.84 1793.37   85.84 1834.66   89.84 2483.49   93.84
#Mann= 2 ,-1 , 0
       0     .06       0  644.92    .035       0
Bank Sta=931.52,1201.91
XS Rating Curve= 0 ,0
Exp/Cntr=0.3,0.1

Type RM Length L Ch R = 1 ,54372.  ,546.44,511.64,507.83
XS GIS Cut Line= 3
 6427277.5682283 2048509.1642128 6427050.5522465  2049543.347972
 6427151.4482542 2050745.6917439
#Sta/Elev= 30
       0   88.55   272.5   85.84  322.13   83.84  397.18   75.78  537.56   71.49
  585.86   65.84   695.4   59.84  738.57   52.25  846.59      44   873.1   35.94
  915.26   34.69  942.39   36.88  968.06    34.6   997.4   37.68 1011.91   43.84
 1016.43   49.84 1019.17   53.84  1032.9   57.84 1084.48   59.07 1165.01   58.92
  1182.3   57.84 1205.99   51.84 1224.45   53.84 1295.57   51.84 1346.32   65.84
 1370.43   67.84 1631.64   73.84 1666.55   81.84  1730.1   85.35 2265.38   91.84
#Mann= 2 ,-1 , 0
       0     .06       0  397.18    .035       0
Bank Sta=738.57,1016.43
XS Rating Curve= 0 ,0
Exp/Cntr=0.3,0.1

Type RM Length L Ch R = 1 ,53861.  ,555.89,594.15,591.83
XS GIS Cut Line= 4
 6426529.2563725 2048219.0882677 6426604.9283665 2049064.0920894
 6426554.8172644 2049541.7052357 6426634.3563273 2050741.4877495
#Sta/Elev= 30
       0   86.07  494.54   85.84  598.96   62.65  646.41   59.84  912.15   57.84
  935.49    48.8  941.42   45.84  998.17   47.84 1009.56   43.84 1021.54      44
 1039.78   35.34 1102.46   34.07 1113.04   36.31 1142.53   34.83 1173.21    37.5
 1187.73   43.84 1200.46   53.84 1207.03   55.36 1227.04   61.84 1432.39   61.41
 1486.23   57.84 1521.25   48.31 1584.26   47.84 1627.34   54.52  1655.9   62.36
 1687.22   65.84 1787.13   69.21 1945.54    82.3 2131.05   87.84 2531.04   90.28
#Mann= 3 ,-1 , 0
       0     .06       0  598.96    .035       0  1655.9     .05       0
Bank Sta=935.49,1207.03
XS Rating Curve= 0 ,0
Exp/Cntr=0.3,0.1

Type RM Length L Ch R = 1 ,53267.  ,630.25,590.58,504.24
XS GIS Cut Line= 5
 6426108.8564589 2048441.9002077 6426041.5924538 2049064.0920894
 6425957.5124711 2049349.9640401  6425974.328496 2049761.9559649
 6426251.7924106 2050863.4037292
#Sta/Elev= 30
       0   85.63  266.22   85.84  315.92   83.84  360.16   73.84  398.28   61.99
  603.91   57.84   625.4   53.79  649.39   43.84  658.46   42.04   668.3      44
  693.56   34.43  705.05    36.2  724.41   33.75  816.07    37.5  851.85   47.84
  918.12   51.75  977.78   61.84 1009.03   63.84 1216.47   63.84 1402.24   57.84
 1431.57   47.84 1480.59   47.84 1501.93   49.84 1509.62   53.84 1533.58   59.84
 1569.86   63.81 1734.25   73.84 1765.38   81.84 1813.22   85.84 2471.99   89.94
#Mann= 3 ,-1 , 0
       0     .06       0  398.28    .035       0 1569.86     .05       0
Bank Sta=625.4,918.12
XS Rating Curve= 0 ,0
Exp/Cntr=0.3,0.1

Type RM Length L Ch R = 1 ,52676.  ,918.25,817.87,500.81
XS GIS Cut Line= 3
 6425402.5845945 2048475.5322103 6425425.3863237 2048984.3236919
 6425530.8065895 2050651.1017515
#Sta/Elev= 30
       0   83.99  187.78   85.84  319.81   83.84  346.12   73.84  362.02   63.84
  390.52   57.81  498.09   53.84  519.21   51.84  524.33    46.9  527.37   43.84
  543.08    44.4  561.64    34.1  571.55    35.6  606.83    33.3  656.56   37.42
  658.55   41.84     673   49.19  701.91   51.16  844.56   47.84  864.57   52.06
  883.15   55.84  1002.8   61.84 1192.92   63.84 1300.31   63.84 1535.47   53.84
 1587.59   53.84 1633.95   58.51 1784.64   69.84  1890.9   83.84 2179.41   85.16
#Mann= 3 ,-1 , 0
       0     .06       0  390.52    .035       0 1633.95     .06       0
Bank Sta=524.33,864.57
XS Rating Curve= 0 ,0
Exp/Cntr=0.3,0.1

Type RM Length L Ch R = 1 ,51858.  ,369.66,361.37,403.21
XS GIS Cut Line= 4
 6424427.2568044 2048853.8921325 6424486.6384679 2049131.0030281
 6425058.6879595  2049835.063908 6425183.9766489 2050787.7317353
#Sta/Elev= 30
       0   79.84  127.37   81.84  375.14   81.84  414.78   73.84  424.56   63.84
  436.58   53.84  513.59    47.5  532.96    46.2  604.89   36.06  693.67   35.22
  719.72   36.23  760.25   49.84  773.84   50.55  825.44   53.84  859.88   57.84
  981.73   61.84 1028.01   61.84 1064.67   63.84 1282.73   63.84 1454.51   57.84
 1483.07   51.84 1551.55   51.84 1578.89   51.84 1639.56   59.84 1683.44   61.84
 1707.94   66.45 1754.94   67.84 1775.07   71.84 1881.39   83.84 2151.43    84.9
#Mann= 3 ,-1 , 0
       0     .06       0  513.59    .035       0 1551.55     .05       0
Bank Sta=532.96,773.84
XS Rating Curve= 0 ,0
Exp/Cntr=0.3,0.1

Type RM Length L Ch R = 1 ,51497.  ,586.49,625.8,619.09
XS GIS Cut Line= 4
 6424027.8769101 2049188.1100899 6424523.9487703 2049734.6299303
 6424692.1087357 2050045.7258948 6424935.9406951 2050802.4457394
#Sta/Elev= 30
       0   81.84   387.8   81.84  435.52   77.84  448.15   73.84  468.06   60.62
  481.04   53.12  513.99   43.84  557.14    35.5  702.51   36.59  725.62   43.84
  747.71    53.7   782.7   55.84   820.3   61.84  892.88   63.84 1112.35   63.84
 1230.93   59.84 1279.34   55.84 1300.47   51.84 1325.72   51.84 1403.11   51.84
 1465.25   59.84 1506.13   59.84 1535.59   63.36  1564.6   63.84  1581.8   65.84
 1600.86   71.84 1661.48   73.84 1704.37   77.93 1741.88   83.84 1886.76   84.17
#Mann= 3 ,-1 , 0
       0     .06       0  468.06    .035       0 1325.72     .05       0
Bank Sta=481.04,747.71
XS Rating Curve= 0 ,0
Exp/Cntr=0.3,0.1

Type RM Length L Ch R = 1 ,50871.  ,342.18,353.62,362.71
XS GIS Cut Line= 3
 6423401.2113233 2049145.6709759 6424105.2722033 2050260.4340161
 6424637.4567612 2051302.7216413
#Sta/Elev= 30
       0   89.13  679.88   91.84  711.97   85.84  728.91   85.84   750.8   83.84
  766.35   73.84  788.33   63.84  826.02   57.77   850.3   53.84  889.19   51.33
 1003.08   43.84 1015.56   38.24  1025.5   35.55 1056.43    37.4 1109.24    36.6
 1138.11   37.62 1157.38   53.06 1221.15   61.84 1243.95   62.24 1372.38   61.84
  1431.6   59.84 1473.29   56.07 1731.29   55.84 1773.29   59.84 1794.96   63.84
 1957.12   69.84 2008.97   73.84  2172.9   79.84 2215.36   83.84 2488.78   83.84
#Mann= 3 ,-1 , 0
       0     .06       0  889.19    .035       0 1473.29     .05       0
Bank Sta=826.02,1157.38
XS Rating Curve= 0 ,0
Exp/Cntr=0.3,0.1

Type RM Length L Ch R = 1 ,50517.  ,524,515.69,513.12
XS GIS Cut Line= 2
 6423269.1999349 2049541.7052357 6424322.1568496 2051357.3736159
#Sta/Elev= 30
       0   89.74  426.42   88.96  469.49   87.84  486.52   83.84   523.2   63.84
  567.18   58.88  588.22   56.55  676.23   45.57  718.95   36.18  732.39   37.61
  753.34   37.21  763.38   38.83  816.71   36.63  853.97   36.69  862.92   43.84
  876.18   48.92  889.26   53.84  944.34   56.32   973.1   61.84 1191.62   59.63
  1404.4   57.89 1503.43   63.84 1517.71   65.84 1633.72   67.84 1767.57   73.84
 1871.89   76.01 1895.45   77.84 1902.41   79.84 1972.55   81.84  2098.9   82.67
#Mann= 3 ,-1 , 0
       0     .06       0  588.22    .035       0 1191.62     .05       0
Bank Sta=567.18,876.18
XS Rating Curve= 0 ,0
Exp/Cntr=0.3,0.1

Type RM Length L Ch R = 1 ,50002.  ,605.1,606.38,615.94
XS GIS Cut Line= 4
 6422909.6131209 2049810.3019242 6423034.5129591 2050172.4264239
  6423533.222759 2051008.4986923 6423850.0686556 2051763.2566727
#Sta/Elev= 30
       0   88.87  294.99   89.84  323.55   85.84  402.13   85.84  417.61   89.84
   474.9   87.91  525.46   73.84  535.68   63.84  563.29   50.74  574.23   43.84
  611.27   41.53  635.24   37.58  650.17      39  670.08      37  685.94   43.84
  747.11   43.84  769.94    35.5   802.9   35.39  819.51   45.84  844.21   47.62
  854.04   45.84 1007.63   45.84 1025.45   47.84 1054.79   55.84 1104.77   59.84
  1126.4    63.6 1155.89   73.84 1160.79   73.84 1677.44   75.84 2175.14   81.01
#Mann= 3 ,-1 , 0
       0     .06       0   474.9    .035       0 1160.79     .05       0
#Block Obstruct= 1 ,-1
 1400.33 2175.14      90
Bank Sta=563.29,844.21
XS Rating Curve= 0 ,0
Exp/Cntr=0.3,0.1

Type RM Length L Ch R = 1 ,49395.  ,422.01,457.34,543.03
XS GIS Cut Line= 2
 6422433.1276665 2050333.7737079  6423407.787002 2052006.8914848
#Sta/Elev= 30
       0   87.84  159.55   87.84  243.45   87.84  257.58   84.04  284.72   82.32
   321.6   73.84  340.62   70.92  374.56   63.84  400.29   54.23   439.3   43.84
  452.73   43.41  474.15    39.1  484.98   39.17  498.04   38.53  548.37   35.21
  581.44    36.7  603.93   34.52  625.45    39.3  642.76   44.59  649.78   45.84
  715.99   45.84  767.15   47.84  907.36   63.84  936.47   73.84 1358.85   75.84
 1637.32   77.84 1724.07   77.84 1790.05   78.42 1822.24   79.84 1936.31   80.53
#Mann= 4 ,-1 , 0
       0     .05       0  159.55     .06       0  400.29    .035       0
  649.78     .06       0
#Block Obstruct= 1 ,-1
 1153.71 1936.31      90
Bank Sta=400.29,642.76
XS Rating Curve= 0 ,0
Exp/Cntr=0.3,0.1

Type RM Length L Ch R = 1 ,48938.  ,408.28,405.47,400.31
XS GIS Cut Line= 4
 6422154.4368946  2050597.796532 6422418.4597187 2051360.5291086
  6422497.621196 2051760.9575046 6422884.3891544 2052618.5733568
#Sta/Elev= 30
       0   87.84   76.05   87.84  108.99   85.84  154.99   73.84  194.81   66.73
  262.43   55.84  293.91   53.84  303.35      50  327.99      41  333.77      37
  351.76   35.03  361.13   43.84  406.41   43.84  417.47    36.3  463.71    34.5
  483.82   35.67  512.31    35.1  530.22      42  541.35   43.84  545.91   48.23
  549.39   51.84  557.32    54.2  563.34   57.49  571.63   57.27  600.19   51.84
   638.1   51.84  656.29   55.84  723.12   63.84   754.3   73.84 2156.11   79.91
#Mann= 3 ,-1 , 0
       0     .06       0  293.91    .035       0  571.63     .05       0
#Block Obstruct= 1 ,-1
  814.71    3000      90
Bank Sta=303.35,545.91
XS Rating Curve= 0 ,0
Exp/Cntr=0.3,0.1

Type RM Length L Ch R = 1 ,48532.  ,306.78,323.87,317.24
XS GIS Cut Line= 3
 6421749.3093876 2050676.3257653 6422085.6293185 2051626.4295417
 6422758.2691804 2052727.8773059
#Sta/Elev= 30
       0   85.98   75.95   83.84  119.31   76.28  194.15   63.84  319.64   54.38
  325.88   53.84  376.73   43.84  383.32   41.51  386.02      40  413.31      35
  429.92   36.01  489.98   34.06  526.88    34.8  550.34      36  572.09   41.99
  576.06   42.52  586.08   43.84  596.03   49.84  624.12   51.02   675.6   51.84
  691.58   53.84  749.02   63.84  776.72   71.84  820.81   73.63   904.6   73.84
 1636.71   75.84 1806.29   77.84 2022.38   77.84 2227.77   79.84 2298.47   80.01
#Mann= 3 ,-1 , 0
       0     .05       0  119.31    .035       0   904.6     .06       0
#Block Obstruct= 1 ,-1
  911.63    3000      90
Bank Sta=319.64,576.06
XS Rating Curve= 0 ,0
Exp/Cntr=0.3,0.1

Type RM Length L Ch R = 1 ,48209.  ,395.02,514.47,823.64
XS GIS Cut Line= 5
 6421480.2534145 2050541.7978024 6421539.1094308 2051046.2776514
 6421698.8614075  2051466.677565 6421934.2853307 2052189.7654544
 6422548.0692235 2052820.3652775
#Sta/Elev= 30
       0   85.52  222.22   83.84  342.28   63.84  360.51   63.42  427.99   61.84
   449.8   57.84  509.02   55.02  542.94   53.84  573.56   43.84  596.37      34
  607.89   35.66  672.58      34   729.3      36  770.69   43.25  776.06   43.84
  790.77   49.41  798.89   53.84  811.41   55.84  940.83   55.84 1170.63   59.26
 1283.61   59.55 1351.42   56.95 1613.09   59.21 1676.57   59.31 1725.03   57.84
 1731.82   59.84 1760.62   63.84  1801.3   73.84 2215.91   77.78 2598.07   79.84
#Mann= 3 ,-1 , 0
       0     .05       0  360.51    .035       0 1170.63     .06       0
#Block Obstruct= 1 ,-1
 1941.34    3000      90
Bank Sta=509.02,770.69
XS Rating Curve= 0 ,0
Exp/Cntr=0.3,0.1

River Reach=Tule Creek      ,Tributary
Reach XY= 30
 6426446.7600056 2059279.8400007 6426252.0299814 2059238.5299987
 6425862.5599927 2058990.6900088  6425154.430021 2058949.3800068
 6424823.9699798 2058819.5600064 6424328.2800126 2058825.4599882
 6423714.5700085 2058677.9300076 6423419.5199875 2058524.4999978
 6423242.4800158  2058329.770021 6422773.3499778 2058146.8300201
 6422307.1600142 2057839.9799882  6421781.969996 2057639.3399946
 6421427.9099803 2057314.7799825 6421183.0100174 2056429.6199793
 6421354.1400199 2056093.2600036 6421265.6300215 2055810.0099935
 6421448.5599875 2055261.2100133 6421498.7199859 2054771.4199805
 6421256.7699903 2054163.6100056 6420861.4000199  2053762.340006
 6420613.5599827 2053343.3700138 6420584.0499916 2053154.5299838
 6420616.5099972 2052888.9800137 6420728.6300049 2052676.5499968
  6420716.829994 2052464.1099923 6420781.7400179 2052334.2800044
 6421041.3900062 2052233.9699952 6421224.3200195 2052045.1300125
 6421513.4700114 2051466.8299814 6421540.4499851 2051194.1899983

Type RM Length L Ch R = 1 ,10982.  ,636.51,604.91,581.58
XS GIS Cut Line= 4
 6425301.0159667 2058105.2966476 6425193.3936153   2058368.97147
  6424945.250402 2058960.2052628  6424775.600164 2059535.5812185
#Sta/Elev= 30
       0   94.35  372.47   93.84  473.56   73.84  492.26   71.84  506.95   69.84
  539.42   67.84  753.42   67.84  759.13   65.54  763.15   63.84  781.68   53.84
  793.75   49.84  803.99   41.82   807.8    38.4  825.67      38  832.01   49.84
  843.33   53.84   856.7    60.1  867.53   64.29  875.58   66.73  897.89   73.84
  914.71   75.84  926.57   77.84  941.89   79.84  975.64   83.84  985.88   85.84
 1025.79   89.84 1033.07   89.84 1040.95   91.84 1066.96   95.84 1525.85   95.28
#Mann= 3 ,-1 , 0
       0     .05       0  759.13    .035       0  875.58     .06       0
Bank Sta=763.15,867.53
XS Rating Curve= 0 ,0
Exp/Cntr=0.3,0.1

Type RM Length L Ch R = 1 ,10377.  ,742.36,780.89,792.31
XS GIS Cut Line= 4
 6424461.5614271  2058121.440005 6424396.9879973 2058734.8875878
 6424380.8446399 2058901.7022655  6424246.316677 2059434.4330138
#Sta/Elev= 30
       0   90.96  211.25   83.84  237.92   83.84  257.05    82.2  333.03   73.84
  346.43   71.28  373.74   67.84  417.12   63.73  471.65   61.42  524.71   61.41
  566.53   62.26  608.16   63.84  615.71   65.84  641.38    65.5  660.86   63.84
  677.15   57.63  687.15   53.84  695.62   49.84   702.1   38.37  717.18    37.6
  725.67   49.84  743.08   53.84  754.73   57.91  771.51   63.84  805.33   73.84
  813.15   77.27  831.45   83.84   905.7   91.35  928.31      95 1333.88      95
#Mann= 3 ,-1 , 0
       0     .06       0  641.38    .035       0  771.51     .05       0
Bank Sta=677.15,754.73
XS Rating Curve= 0 ,0
Exp/Cntr=0.3,0.1

Type RM Length L Ch R = 1 ,9596.   ,483.01,513.72,529.78
XS GIS Cut Line= 4
 6423966.3303657 2057864.4915736  6423794.302716 2058218.3001497
 6423735.1103896 2058379.7337241 6423482.8704414 2059083.6513232
#Sta/Elev= 30
       0   93.84  127.52   93.84  377.21   84.29  392.57   83.84  432.43   83.84
  467.07    82.2  557.18   73.84  636.52   63.84  669.52   61.84  684.47   59.84
  691.54   59.84  735.79   63.84   749.7   65.84  777.08   65.84  800.53   63.84
  802.99    62.8  811.25   59.71  826.92   53.84  833.79   49.84     840    38.2
  853.34    37.4  859.65   49.84  892.03   59.96   905.8   63.84  920.38   72.59
  923.09   73.84  932.34   82.22  933.52   83.84  1094.8   86.43  1313.1   91.88
#Mann= 3 ,-1 , 0
       0     .05       0  802.99    .035       0   905.8     .06       0
Bank Sta=811.25,892.03
XS Rating Curve= 0 ,0
Exp/Cntr=0.3,0.1

Type RM Length L Ch R = 1 ,9082.   ,471.53,468.89,465.86
XS GIS Cut Line= 4
 6423608.9904155 2057717.3516275 6423419.9516762    2058029.6771
 6423055.4148794 2058653.2268603 6422915.3305816 2058926.0013674
#Sta/Elev= 30
       0   93.29   27.07   93.84  329.83   93.84  360.36    92.6  407.58   91.84
  463.55   81.72  513.71   73.84  552.89   63.84  580.03   59.84  597.67   59.84
  635.25   65.84  655.76   65.84  666.74   63.84  672.61   60.09  679.85   55.47
  683.64   53.84  700.31   49.84  710.79      38  721.36    37.2  727.19   49.84
  748.84   54.61   770.3   60.13  788.34   63.84  810.21   72.57  821.22   73.84
  912.16   73.84  952.53   81.66  958.98   83.84 1164.36      95 1394.01      95
#Mann= 3 ,-1 , 0
       0     .06       0  655.76    .035       0  810.21     .05       0
Bank Sta=672.61,748.84
XS Rating Curve= 0 ,0
Exp/Cntr=0.3,0.1

Type RM Length L Ch R = 1 ,8613.   ,552.42,559.35,555.17
XS GIS Cut Line= 4
 6423188.5905018   2057444.09166  6422852.606881 2058078.3910834
 6422734.2222756 2058315.1602943  6422421.360695 2058841.9213847
#Sta/Elev= 30
       0   93.84  306.03   93.84  420.86   91.84  435.08   83.84   461.7   73.84
  549.23   61.84  564.32   63.84  598.72   59.84  616.56   59.84  630.94   61.84
  639.68   63.84  720.57   65.84  765.34   65.84   770.3   64.52  773.25   62.93
  790.54   53.84  804.33   49.84  807.11   41.96  808.32    37.8  815.39      37
   820.8   49.84   832.9   53.84  845.19   56.96  870.34   63.84  880.96   65.69
  941.66   74.07 1004.73   83.84 1023.23   85.45 1286.68   93.37 1595.17   92.74
#Mann= 3 ,-1 , 0
       0     .05       0  765.34    .035       0  880.96     .06       0
Bank Sta=773.25,845.19
XS Rating Curve= 0 ,0
Exp/Cntr=0.3,0.1

Type RM Length L Ch R = 1 ,8054.   ,372.38,388.69,382.15
XS GIS Cut Line= 4
 6422684.1106055 2057307.4617236 6422384.4495626 2057782.4295461
 6422309.1138787 2057938.4819698 6422021.9807533 2058389.9914893
#Sta/Elev= 30
       0   93.84   84.27   93.84   256.3   91.84  288.39   87.84  292.29   86.42
  358.19   73.84  385.49   67.84  391.92   61.84  400.15   63.84   433.5   61.47
  446.45   59.84  505.98   59.84   528.9   63.84  550.03   63.84  583.23   58.39
  610.18   54.52  614.92   53.84  626.61    50.3  639.86   47.84  653.55   37.61
   662.7   36.89  675.78   47.84  681.74   50.98  714.61   65.35  729.04   73.84
  738.44   83.84   752.5   87.84  817.55   89.84  858.88   91.84 1269.96   90.29
#Mann= 3 ,-1 , 0
       0     .06       0  583.23    .035       0  714.61     .05       0
Bank Sta=610.18,681.74
XS Rating Curve= 0 ,0
Exp/Cntr=0.3,0.1

Type RM Length L Ch R = 1 ,7665.   ,483.42,518.81,532.63
XS GIS Cut Line= 4
  6422298.351672 2057233.5553931  6422050.820207 2057620.9959717
 6421943.1978083  2057814.716261 6421679.5229859 2058137.5833625
#Sta/Elev= 30
       0   92.24   79.65   91.84  101.28   83.84  104.48   83.39  144.38   83.18
  158.37   81.84  212.64   71.27  232.72    65.8  235.69   61.84  274.77   63.84
  301.93   61.84  437.77   59.84  458.09   63.84  462.73   63.84  486.23   59.18
  512.28   53.84  541.22   49.42  554.23   47.84  577.15    38.9  602.47    36.8
  611.58    38.6  623.14   50.85  626.44   53.84  643.83   63.84  657.06   73.84
  682.52   82.52   706.5   85.84  708.96   87.84  723.58   91.84 1098.23   90.74
#Mann= 3 ,-1 , 0
       0     .05       0  486.23    .035       0  626.44     .06       0
Bank Sta=541.22,623.14
XS Rating Curve= 0 ,0
Exp/Cntr=0.3,0.1

Type RM Length L Ch R = 1 ,7146.   ,455.16,511.54,541.53
XS GIS Cut Line= 3
 6422040.0579529 2056980.6428247 6421728.8845969 2057259.9288252
 6421259.7957397 2057793.1917528
#Sta/Elev= 30
       0   91.84   26.43   87.57    63.7   85.84   73.29   83.84  105.77   83.84
  209.38   77.84  229.86   75.84  240.48   73.84  244.79    71.1  268.25   61.84
  549.94   63.84  580.59   59.84  612.05   55.84  626.96   51.85  638.42   47.84
  646.58    38.9  654.01    37.5  669.29    36.8  677.42    38.6  682.61   47.84
  712.48   53.91  737.77   60.14  775.75   67.84  793.62   69.84  857.38   79.59
  980.94    84.7 1000.45   85.84 1010.93   87.84 1091.54   91.84 1128.35   91.84
#Mann= 3 ,-1 , 0
       0     .06       0  580.59    .035       0  712.48     .05       0
Bank Sta=626.96,712.48
XS Rating Curve= 0 ,0
Exp/Cntr=0.3,0.1

Type RM Length L Ch R = 1 ,6635.   ,348.69,362.82,378.39
XS GIS Cut Line= 4
 6421874.8408072 2056802.9818272 6421577.2817378 2056894.5449342
 6421200.6034133 2057066.7407153 6420750.2710501  2057475.621689
#Sta/Elev= 30
       0   91.84   92.22   91.84  108.77   90.71  238.06   91.84  243.51   89.84
   262.5   89.84  277.61   91.81  311.33   90.51  341.99   85.84  388.64   75.84
  446.11   73.84  501.62   63.84  542.06   53.84  555.99   50.37  574.84   45.84
  581.73    38.9  601.16    36.7  608.81    38.6  613.36   45.84  625.22   54.15
  637.39   55.84  660.24    56.6   676.3   63.84   705.6   67.84  892.54   71.84
  903.74   73.84 1008.66   77.84  1210.7   83.84 1259.33   83.84 1333.76   90.07
#Mann= 3 ,-1 , 0
       0     .05       0  542.06    .035       0  637.39     .06       0
Bank Sta=555.99,625.22
XS Rating Curve= 0 ,0
Exp/Cntr=0.3,0.1

Type RM Length L Ch R = 1 ,6272.   ,424.48,491.73,562.7
XS GIS Cut Line= 4
 6421785.2956081 2056601.2739249 6421338.6627505 2056628.1795364
 6421053.4634199  2056714.277427 6420597.4136432 2056915.0604174
#Sta/Elev= 30
       0   91.84  282.04   91.84  426.04   73.84  447.11   69.22  516.28   57.84
   529.3   55.84  538.51   53.02  549.62   45.84  554.92   43.54  560.66    38.9
  579.88    36.5   585.8    38.6  592.83    43.9  599.89   45.84  607.37   51.54
  610.41   53.84  628.67   57.84  636.29   59.84  656.12   61.84  662.61   63.84
  852.21   65.84  906.82   67.84  928.57   73.84  984.62    74.9 1013.08   77.84
 1110.71   83.84 1134.39   87.84 1143.53   91.07 1149.79   91.84 1243.65   91.84
#Mann= 3 ,-1 , 0
       0     .06       0  516.28    .035       0  628.67     .05       0
Bank Sta=538.51,607.37
XS Rating Curve= 0 ,0
Exp/Cntr=0.3,0.1

Type RM Length L Ch R = 1 ,5780.   ,445.59,455.6,394.01
XS GIS Cut Line= 4
 6422059.7326846 2056246.1201085 6421403.2361802 2056240.7389578
 6421182.6102794 2056170.7844247 6420730.5963184 2056036.2564618
#Sta/Elev= 30
       0   89.84   31.47   89.84   50.35   91.84  282.07   91.84  410.79   89.84
  427.39   87.84  468.16   79.84  509.92   77.84  530.53   69.84  597.29   67.84
  682.58   67.84  690.35   65.84  698.03   63.84  715.42   53.84  729.83   49.86
  742.97   45.84  755.13    38.8  774.53    36.3  778.48    38.4  782.68    43.7
  807.72   52.92  829.14   61.84 1030.52   63.84 1050.95   67.84 1110.13   69.84
 1125.99   73.84 1179.24   78.92 1215.62   87.84 1273.36   91.84 1359.58   91.84
#Mann= 3 ,-1 , 0
       0     .05       0  690.35    .035       0  829.14     .06       0
Bank Sta=729.83,807.72
XS Rating Curve= 0 ,0
Exp/Cntr=0.3,0.1

Type RM Length L Ch R = 1 ,5325.   ,360.91,397.41,407.35
XS GIS Cut Line= 4
 6422059.7326846 2055815.6306083 6421636.7911093 2055810.9909965
 6421214.8969943 2055777.9627427 6420843.5998205 2055708.0082096
#Sta/Elev= 30
       0   87.84   24.29   89.84  198.86   89.84  231.66   87.84  307.65   85.84
  339.44   80.26  377.82   71.84  553.86   67.84  598.21   69.84  645.27   69.84
  652.27   65.84  717.13   63.84  738.97   53.84   748.5   51.05  775.94      43
  778.55    38.5  790.67    36.2  797.84    38.2  804.14    43.5  810.36   45.84
  819.71   52.48  846.79   61.84  895.11   63.84  906.51   65.84  934.64   73.84
  966.88   75.84 1006.41   83.84 1056.62   87.84    1160   89.84 1223.98   89.84
#Mann= 3 ,-1 , 0
       0     .06       0  717.13    .035       0  846.79     .05       0
Bank Sta=748.5,819.71
XS Rating Curve= 0 ,0
Exp/Cntr=0.3,0.1

Type RM Length L Ch R = 1 ,4927.   ,232.92,240.23,246.74
XS GIS Cut Line= 4
  6422022.064819  2055568.099096 6421518.9302103 2055447.0239625
 6421231.0403517 2055358.2354966 6420940.4599651 2055336.7109884
#Sta/Elev= 30
       0   81.47      45   79.84  192.14   80.12  241.93   81.16  257.56   79.84
   288.7   79.84  315.02   77.84  358.01   71.84  521.59   71.23  576.47   69.52
  593.36   63.84   599.3   53.84  605.98   50.99   625.7   42.73   631.7   38.41
  647.57   36.02  653.69   38.01  660.77      43  669.53   45.84  676.98   47.05
  734.55   53.84  753.13   59.77  769.72   63.84   796.8   73.84  815.56   77.84
  852.67   79.84  891.89   87.84  966.67   87.84  984.41   85.84 1110.14   85.84
#Mann= 3 ,-1 , 0
       0     .05       0  576.47    .035       0  734.55     .06       0
Bank Sta=605.98,676.98
XS Rating Curve= 0 ,0
Exp/Cntr=0.3,0.1

Type RM Length L Ch R = 1 ,4687.   ,327.57,321.23,302.9
XS GIS Cut Line= 4
 6422200.8209899   2055280.37131 6421532.3830398  2055218.326383
 6421353.3866947 2055142.5356273 6420950.0896518 2055106.8004206
#Sta/Elev= 30
       0    88.2   28.26   87.84   49.14   81.84   63.88   75.84   185.6   73.84
  214.33   71.84  346.22   69.84  418.14   69.84  470.88   71.84  479.78   73.84
  696.38   73.84  711.58   69.84   716.1   67.68  723.69   63.84  740.47   52.18
  752.87   43.84  762.43    42.7   771.4    38.4  790.17    35.8   797.8      38
  805.88      43  816.49   43.84  840.93   48.68  848.88   49.84  865.69   54.67
   895.7   63.63  912.08   74.35  938.84   83.84 1015.76   85.15 1270.57   85.84
#Mann= 3 ,-1 , 0
       0     .05       0  740.47    .035       0  865.69     .06       0
#XS Ineff= 2 ,-1
       0     700      78     900 1270.57      85
Permanent Ineff=
       F       F
Bank Sta=740.47,840.93
XS Rating Curve= 0 ,0
Exp/Cntr=0.3,0.1

Type RM Length L Ch R = 3 ,4514.   ,,,
Node Name=Yosemite Street
Bridge Culvert--1,0,-1,-1, 0
Deck Dist Width WeirC Skew NumUp NumDn MinLoCord MaxHiCord MaxSubmerge Is_Ogee
100,96,2.6,0, 68, 68, , , 0.95, 0, 0,0,,
       0   15.84   38.96   47.45   52.19   54.37   55.98   58.77   62.42   68.02
   71.18    82.9   92.33    96.7  118.56  127.25  140.33  150.82  152.09  155.23
   180.5  189.97  207.31  219.58  236.79  238.37  243.91   247.2  256.83  260.81
  263.15  276.94  287.04  294.83  299.52  308.71  309.17  315.37  319.48  320.32
  329.13  331.76  340.19  345.44  352.11  359.42  363.77  373.26  374.58  382.66
  382.75  383.33  398.14  412.47  416.47  419.25  427.98  432.98  441.15  451.21
  460.76  466.12     525     725     725     875     875    1200
   88.73    88.7   88.15   87.84   87.84   86.75   85.84   84.96   83.84   82.55
   81.84   78.56   75.84   75.65   75.14   74.93   74.91   74.03   73.84   73.84
   73.84   73.84   73.84   73.84   73.84   73.47   72.79   72.86   73.45    73.7
   73.84   74.76   75.05   75.26   75.48   75.69   75.71   75.84   76.01   76.04
   76.39   76.47   76.58   76.75   76.85   77.12    77.2   77.62   77.64   77.83
   77.83   77.84   77.91   77.99   77.84   77.84   76.99   77.02   76.96    76.2
   76.17   76.21      78      84      84      84      84      84
                                                                                
                                                                                
                                                                                
                                                                                
                                                                                
                                                                                
                                      74      74
       0   15.84   38.96   47.45   52.19   54.37   55.98   58.77   62.42   68.02
   71.18    82.9   92.33    96.7  118.56  127.25  140.33  150.82  152.09  155.23
   180.5  189.97  207.31  219.58  236.79  238.37  243.91   247.2  256.83  260.81
  263.15  276.94  287.04  294.83  299.52  308.71  309.17  315.37  319.48  320.32
  329.13  331.76  340.19  345.44  352.11  359.42  363.77  373.26  374.58  382.66
  382.75  383.33  398.14  412.47  416.47  419.25  427.98  432.98  441.15  451.21
  460.76  466.12     525     725     725     875     875    1200
   88.73    88.7   88.15   87.84   87.84   86.75   85.84   84.96   83.84   82.55
   81.84   78.56   75.84   75.65   75.14   74.93   74.91   74.03   73.84   73.84
   73.84   73.84   73.84   73.84   73.84   73.47   72.79   72.86   73.45    73.7
   73.84   74.76   75.05   75.26   75.48   75.69   75.71   75.84   76.01   76.04
   76.39   76.47   76.58   76.75   76.85   77.12    77.2   77.62   77.64   77.83
   77.83   77.84   77.91   77.99   77.84   77.84   76.99   77.02   76.96    76.2
   76.17   76.21      78      84      84      84      84      84
                                                                                
                                                                                
                                                                                
                                                                                
                                                                                
                                                                                
                                      74      74
BR Coef=-1 , 0 , 0 ,, 0 ,,,0.8,0,,0,
WSPro=,,,, 1 ,,,, 0 ,,,, 0 ,,,,-1 ,-1 ,-1 , 0 , 0 , 0 , 0 , 0
BC Design=,, 0 ,, 0 ,,,,,,
BC HTab HWMax=95
BC HTab MaxFlow=10000
BC Use User HTab Curves=0
BC User HTab FreeFlow(D)= 0

Type RM Length L Ch R = 1 ,4366.   ,356.48,320.19,265.47
XS GIS Cut Line= 5
  6422256.976254 2055050.6451565 6421889.4144178 2055004.6998974
 6421634.1631098  2054907.704424 6421332.9665901 2054826.0240055
 6420893.9343877 2054815.8139531
#Sta/Elev= 30
       0   88.32   15.65   87.84   78.09   87.84   89.64   88.39  161.84   87.84
  342.96   83.03  350.11   81.84  464.24   78.22  684.19   75.84     705   74.49
  718.53   71.84  748.43   60.45  764.81   53.03  779.88   43.84  792.85   42.53
   800.1    38.2  819.32    35.6  824.94    37.8  831.13   42.58  842.68   43.84
  857.29   53.07  867.79   59.23  894.48   73.84  906.64   75.84  920.82   79.84
  926.51   80.49  953.56   81.46 1159.86   81.75 1197.76   82.99 1394.71   83.84
#Mann= 3 ,-1 , 0
       0     .06       0  748.43    .035       0  867.79     .05       0
#XS Ineff= 2 ,-1
       0  706.56      81     900 1394.71   83.84
Permanent Ineff=
       F       F
Bank Sta=764.81,857.29
XS Rating Curve= 0 ,0
Exp/Cntr=0.3,0.1

Type RM Length L Ch R = 1 ,4046.   ,256.61,245.09,234.47
XS GIS Cut Line= 4
  6421940.591346 2054474.6389447 6421579.4678244 2054505.3281276
 6421283.5062871 2054612.9505263 6420792.4791728 2054774.3841007
#Sta/Elev= 30
       0   89.16  292.39   87.84  327.19   85.84  421.91   85.84   434.7   83.84
  448.62   73.84  477.12   63.84   500.2   53.84   500.4   53.63  509.84   43.84
  516.31      42  524.92      38  531.08    36.2  538.55    35.4   546.8    37.4
  556.46    42.5  573.47   43.84  578.09    46.7   587.8   53.84  612.22   63.84
  631.25   71.19  636.24   73.84  655.63   74.94  670.69   74.53  687.56   75.39
  702.05   78.37  789.23   80.77 1096.53   83.84 1164.68   85.84 1194.23   85.84
#Mann= 3 ,-1 , 0
       0     .05       0   500.2    .035       0  612.22     .06       0
#XS Ineff= 2 ,-1
       0  128.5289.16025  690.55 1194.23   85.84
Permanent Ineff=
       F       F
Bank Sta=500.4,578.09
XS Rating Curve= 0 ,0
Exp/Cntr=0.3,0.1

Type RM Length L Ch R = 1 ,3801.   ,152.9,161.27,167.29
XS GIS Cut Line= 5
 6421727.4485694 2054269.9042043  6421424.760641 2054283.3569864
 6421209.5158909 2054397.7057762 6421108.6199306 2054471.6961723
 6420765.5735613 2054619.6769173
#Sta/Elev= 30
       0    88.4  171.37   87.84  280.35   83.84  294.02   81.84  315.03   80.92
  324.96   80.97  333.26   79.84  340.13   77.84  348.97   73.84  361.53   63.84
  376.08   55.27  378.57   53.84  393.48   47.61  404.59   43.84  411.55      42
  418.21      38  427.81    36.2  435.23    35.2  443.14    37.4  451.28    42.5
  461.11   43.84  472.71   52.83  488.02   63.84  533.19   65.84  552.46   67.84
  572.17   73.84  581.68   81.14  586.34   83.84  606.87   85.84 1045.44   85.84
#Mann= 3 ,-1 , 0
       0     .06       0  376.08    .035       0  488.02     .05       0
Bank Sta=376.08,472.71
XS Rating Curve= 0 ,0
Exp/Cntr=0.3,0.1

Type RM Length L Ch R = 1 ,3639.   ,393.56,418.86,402.11
XS GIS Cut Line= 4
 6421749.3093876 2054157.2370123 6421396.1734318 2054132.0129986
 6421076.6695258 2054274.9489976 6420689.9016147 2054485.1489544
#Sta/Elev= 30
       0   88.04   244.9   87.84  323.07   85.77  353.36   83.84  366.09   78.23
  375.14   75.37  416.05   74.98  423.19   73.84  463.37   53.84  468.33   49.37
  474.46   43.84  482.02      42   488.9   37.95  508.66   35.14   515.7    37.2
  524.91   42.38  535.64   43.84  549.71   53.84  555.12   54.33  562.86   55.04
  568.74   55.84  643.46   57.84  668.78   61.84     782   64.47  865.59   67.84
   893.6   71.84  901.47   73.84  912.01   83.84  925.22   85.84 1144.25   85.84
#Mann= 3 ,-1 , 0
       0     .06       0  463.37    .035       0  562.86     .05       0
Bank Sta=468.33,555.12
XS Rating Curve= 0 ,0
Exp/Cntr=0.3,0.1

Type RM Length L Ch R = 1 ,3220.   ,287.29,281.67,325.5
XS GIS Cut Line= 6
 6421816.5733454 2053955.4450443 6421303.6854602 2053787.2850788
 6421076.6695258 2053846.1410952 6420874.8775578 2053963.8530804
 6420689.9016147 2054073.1570296 6420446.0696553 2054224.5010174
#Sta/Elev= 30
       0   87.84  357.18   87.84  362.28   85.69  388.63   83.84  422.13   73.84
  580.87   74.28  589.33   73.84  672.67   63.84  721.64   61.42  781.37   60.99
  806.48   57.84  825.93   53.84  840.03   49.54  858.28   43.84     871      42
  878.22    37.8  903.36    34.9  923.07      42  933.83   43.84  948.66   53.84
  949.93   54.03   962.3   55.84 1007.19   59.84 1244.21   63.84 1304.04   69.84
 1310.82   71.84 1332.54   73.84 1401.29   83.84 1420.33   85.84 1509.73   86.25
#Mann= 3 ,-1 , 0
       0     .05       0  825.93    .035       0   962.3     .06       0
Bank Sta=840.03,949.93
XS Rating Curve= 0 ,0
Exp/Cntr=0.3,0.1

Type RM Length L Ch R = 1 ,2939.   ,109.06,109.27,98.98
XS GIS Cut Line= 5
  6421850.205348  2053795.693115 6421370.9494653 2053635.9411383
 6420992.5895431 2053585.4931582 6420706.7175923 2053728.4291099
 6420235.8696985 2053787.2850788
#Sta/Elev= 30
       0   87.49  266.92   86.67  304.99   81.11  326.61   73.84   387.1   73.84
  510.58   77.84  551.54   78.15  616.21   77.84  693.63   73.67  773.47   73.32
  886.89   75.92  968.65   73.84  983.07   69.84 1015.61   55.64  1033.5   49.31
 1050.53   43.84 1065.35      42 1072.97   37.62  1094.5    34.9 1114.29      42
 1125.47   43.84 1135.11   53.84 1140.83   54.25 1161.11   55.84 1185.96   57.84
 1383.95   61.84 1419.81   63.84 1450.88   67.51 1554.41   85.84 1681.02   87.13
#Mann= 3 ,-1 , 0
       0     .05       0 1015.61    .035       0 1161.11     .06       0
Bank Sta=1033.5,1140.83
XS Rating Curve= 0 ,0
Exp/Cntr=0.3,0.1

Type RM Length L Ch R = 1 ,2830.   ,397.69,471.43,505.66
XS GIS Cut Line= 5
 6421883.8373505 2053703.2050961 6421337.3174628 2053535.0451307
 6420933.7335268 2053493.0051393 6420631.0455984 2053644.3491271
 6420193.8297072 2053694.7971073
#Sta/Elev= 30
       0    86.3  249.24   85.19  259.71   83.84  294.73   73.84   344.7   72.51
  478.23   77.51  581.64   79.84  765.06   78.65  951.79   79.25 1031.55   73.84
 1044.31   71.74 1055.67   69.84 1103.94   53.84 1126.53   47.65 1138.26   43.84
 1151.32      42 1158.91    37.5 1183.13    34.9 1188.88      37 1195.55      42
 1206.24   43.84 1230.26   52.83 1236.34   54.27 1258.15   55.84 1282.96   57.84
 1431.77   61.84 1457.24   63.84 1476.11   65.84 1593.73   85.84 1756.11   87.63
#Mann= 3 ,-1 , 0
       0     .05       0 1103.94    .035       0 1258.15     .06       0
Bank Sta=1126.53,1230.26
XS Rating Curve= 0 ,0
Exp/Cntr=0.3,0.1

Type RM Length L Ch R = 1 ,2358.   ,103.59,92.62,89.23
XS GIS Cut Line= 5
 6422001.5493358 2053291.2132186 6421143.9334836 2053106.2372282
 6420816.0215888 2053165.0932445 6420370.3976614 2053148.2772196
 6420185.4217184 2053148.2772196
#Sta/Elev= 30
       0   84.01  128.06   79.84  146.57   73.84  193.09   73.84  298.79   62.65
  462.39   51.84  545.86   51.84  706.23   65.84  776.13   73.84   849.9   79.84
  885.98    80.2 1111.41   79.57 1242.09   65.84 1384.42   54.33 1388.86   53.84
  1405.9   43.84 1418.87      42 1424.33    37.5 1444.74    34.8 1466.68   43.84
 1476.03   51.83  1478.4   53.84 1499.37   56.03 1552.36   57.84 1590.76   63.84
 1639.27   73.84 1661.44   83.84 1672.04   85.84 1709.67   87.84 1841.41   87.78
#Mann= 3 ,-1 , 0
       0     .06       0 1384.42    .035       0 1499.37     .05       0
Bank Sta=1384.42,1476.03
XS Rating Curve= 0 ,0
Exp/Cntr=0.3,0.1

Type RM Length L Ch R = 1 ,2265.   ,411.11,411.57,375.33
XS GIS Cut Line= 5
 6422018.3653134 2053207.1332359 6421110.3015284 2053005.3412679
 6420706.7175923 2053064.1972369 6420479.7016579 2053064.1972369
 6420193.8297072 2053047.3812592
#Sta/Elev= 30
       0   82.24   117.5   79.84  129.87   73.84  185.08   73.84  197.33   77.42
  265.39   73.02  383.52   72.89  431.73    68.2  541.69   49.84   579.8   49.84
  883.91   77.84  923.15   77.84 1078.96   68.09 1216.93   65.21 1391.05   54.31
 1401.68   50.94 1413.73   43.84  1427.2      42 1431.98    37.5 1455.34    34.8
 1478.85   43.84 1486.94   50.69 1490.62   53.84 1502.92   55.71 1567.57   57.84
 1636.03   67.84 1663.32   73.84 1684.27   83.84 1693.68   85.84 1851.45   87.11
#Mann= 3 ,-1 , 0
       0     .06       0 1391.05    .035       0 1502.92     .05       0
Bank Sta=1401.68,1486.94
XS Rating Curve= 0 ,0
Exp/Cntr=0.3,0.1

Type RM Length L Ch R = 1 ,1854.   ,227.51,258.79,268.52
XS GIS Cut Line= 5
 6422192.0691175 2052963.7118541 6421280.1430916 2052707.6981328
 6420863.1063735 2052687.5189123 6420627.6824029 2052680.7925213
 6420237.9717194 2052814.0593095
#Sta/Elev= 30
       0   80.12   509.1   75.84  533.55   73.84  569.68   63.84  616.54   53.84
  722.57   45.84  947.18   45.76  1063.9   47.84 1112.78   50.22 1203.43   61.84
 1266.44   63.64 1322.94   61.84 1368.57    54.1 1423.26   49.24 1445.12   47.84
 1473.63      42 1487.22    37.2  1508.2    34.6  1516.9      37 1526.04      42
 1535.84   43.84 1555.87   53.84  1560.2    54.4 1582.26    57.2 1707.38   59.84
 1777.26    63.3 1835.51   71.84 1853.62   77.84  1876.6   81.84 2012.09   85.05
#Mann= 3 ,-1 , 0
       0     .06       0 1423.26    .035       0 1582.26     .06       0
Bank Sta=1445.12,1560.2
XS Rating Curve= 0 ,0
Exp/Cntr=0.3,0.1

Type RM Length L Ch R = 1 ,1595.   ,601.62,1595.1,597.12
XS GIS Cut Line= 6
 6422369.1971783 2052943.6596315 6421588.0439919   2052573.50648
 6421098.3621653 2052514.3141536  6420657.110411  2052417.454009
 6420517.2012974 2052460.5029779 6420275.0509832 2052670.3666247
#Sta/Elev= 30
       0   80.22  698.06   75.84  728.81   77.78  796.33   77.84   854.5   73.84
  916.37   63.84 1000.66   63.84 1044.95   61.84  1424.6   61.84 1662.48   57.84
 1682.15   53.84 1687.87    50.3 1698.27   43.84 1707.09      42 1714.27    37.2
 1727.52      35 1738.86    34.6 1747.56   36.97 1757.49      42 1765.68   43.84
 1782.52   53.09 1810.81   59.84  1838.8   61.84 1919.01   65.84 1956.07    65.5
 1992.04   66.65 2078.08   71.65 2206.63   73.84 2239.24   83.84 2276.51   85.26
#Mann= 4 ,-1 , 0
       0     .06       0  1424.6     .05       0 1662.48    .035       0
  1838.8     .06       0
Bank Sta=1687.87,1782.52
XS Rating Curve= 0 ,0
Exp/Cntr=0.3,0.1

River Reach=Baxter River    ,Lower Reach
Reach XY= 30
 6421540.4499851 2051194.1899983 6420055.4399767 2051167.6800068
 6417503.0800234 2050584.2799906 6417277.6799867 2049881.5500087
  6417436.779981 2046765.6799998 6416303.1399811 2045559.1099864
 6415268.9299987 2045002.2299967 6414327.5399906 2044763.5700178
  6413081.199996 2043914.9899963  6411934.290019  2043702.840009
 6411271.3400057 2043835.4399992 6409163.1500126 2043742.6199777
 6406630.6800199 2045466.2999997 6405444.0000144 2046036.4299915
 6404104.8399983 2045917.0999784 6403110.4099846 2045466.2999997
  6401757.989979 2044352.5400203 6399968.0199967 2039738.4000136
 6397674.2099829 2036980.5199967 6396620.1199801 2036251.2699883
 6394551.7100029 2035972.8299935 6393623.5799844 2036251.2699883
 6393172.7700182 2036556.2300096 6392695.4399782 2038147.3099942
 6392005.9800207  2038505.310021  6391369.539999 2038531.8300001
 6390355.2300122 2037908.6500153 6389254.7300223 2035707.6499881
 6388061.4199984 2035323.1400171 6387438.2400136 2035323.1400171

Type RM Length L Ch R = 1 ,47694.  ,157.08,138.01,115.25
XS GIS Cut Line= 5
 6421184.4600559 2050695.4960081 6421130.6488802 2051045.2687211
 6421017.6453781 2051443.4715065 6420377.2922312 2052487.4085894
 6420221.2397601  2052718.796697
#Sta/Elev= 30
       0   84.06   112.4   81.84   153.8   75.84  159.25   73.84   242.4   63.84
  257.29   63.65  316.39   61.84  342.82   57.84  437.24   56.43   463.1   55.84
  473.52   53.84  485.34   43.84  500.14   33.61  515.31   34.95  561.66   33.59
  617.94    34.6  640.78    36.7  675.05      42  697.49   43.84  726.89   53.93
   751.8   59.84 1813.96   59.84 1975.51   61.84 2011.29   65.86 2048.83   71.84
 2117.59   72.53 2141.02   73.84 2171.88   83.84 2216.45   85.84 2271.59   85.84
#Mann= 3 ,-1 , 0
       0     .06       0  257.29    .035       0 2011.29     .05       0
Bank Sta=437.24,726.89
XS Rating Curve= 0 ,0
Exp/Cntr=0.3,0.1

Type RM Length L Ch R = 1 ,47556.  ,188.27,200.04,182.63
XS GIS Cut Line= 5
 6421033.7887356 2050630.9225784 6420963.8342024 2051131.3666117
 6420920.7852335 2051384.2791801 6420242.7642683 2052600.4120442
  6420143.381727 2052744.6933309
#Sta/Elev= 30
       0   84.51   170.5   81.84  240.09   73.84  288.82   63.84  321.97   63.02
  503.05   56.25  522.49   55.84  532.18   53.84   548.4   43.84  552.39   38.55
  561.81   37.57  571.01   33.47  587.71    34.8  640.31   33.42  695.86   34.69
  734.97   43.79  743.14      42  759.52   43.84  774.03   53.84  793.31   59.84
  802.17   59.91 1824.94   59.84 2028.16   61.84 2048.34   65.33 2081.48   70.82
 2142.51   71.84 2161.82   73.84 2191.25   83.84 2222.82   85.84 2329.43   86.98
#Mann= 3 ,-1 , 0
       0     .06       0  321.97    .035       0 2048.34     .05       0
Bank Sta=503.05,802.17
XS Rating Curve= 0 ,0
Exp/Cntr=0.3,0.1

Type RM Length L Ch R = 1 ,47356.  ,211.15,254.47,293.61
XS GIS Cut Line= 6
 6420842.7590216 2050573.7481598 6420775.4950165 2051165.6712344
 6420681.3254472 2051441.4535986 6420479.5334792 2051898.8487103
 6420170.1191598 2052416.7813888 6419901.0631867 2052706.0165351
#Sta/Elev= 30
       0   84.12  264.36   81.84  296.46   75.84  325.14   73.06  357.39   75.84
  378.46   75.84  413.35   75.84  422.63   74.28  445.42   63.84  468.13   59.84
  553.43   56.23  571.18   53.84  610.69   37.43  629.99   34.11   716.2   33.93
  746.18   36.56   765.9   43.43  781.56      42  793.41   43.84  810.59   53.84
  832.77   59.86 1865.78   59.84 2106.71   61.84 2135.66    67.1 2150.59   69.84
 2244.34   71.84 2260.29   73.84 2275.09   78.14 2335.37   87.19 2385.43   87.84
#Mann= 3 ,-1 , 0
       0     .06       0  378.46    .035       0 2135.66     .05       0
Bank Sta=553.43,832.77
XS Rating Curve= 0 ,0
Exp/Cntr=0.3,0.1

Type RM Length L Ch R = 1 ,47102.  ,82.86,82.14,76.88
XS GIS Cut Line= 6
 6420721.6838408 2050560.2953777 6420566.9766574 2051064.7752741
  6420405.543083 2051407.8215961 6420170.1191598 2051851.7639257
 6419921.2424071 2052221.7158118 6419551.2904737  2052645.478921
#Sta/Elev= 30
       0   84.26  309.01   81.95   332.5   75.84  355.06   65.84  364.13   63.84
   407.4    66.4  455.47   69.84  500.91   59.84  551.91   57.84  573.15   54.67
   599.5   43.84  627.88    42.9  637.85    38.4  652.16   35.97  743.02   34.06
  761.92    36.4  773.85   42.96  810.29   43.84  823.08   53.84  834.65   56.78
  846.78   59.84  951.73   60.64 2129.45    60.7 2230.38   61.84 2243.86   63.84
 2261.69   69.84 2295.07   72.41 2312.19   73.84 2387.62   87.84 2417.71   87.91
#Mann= 3 ,-1 , 0
       0     .05       0   407.4    .035       0 2295.07     .06       0
Bank Sta=573.15,834.65
XS Rating Curve= 0 ,0
Exp/Cntr=0.3,0.1

Type RM Length L Ch R = 1 ,47019.  ,509.62,485.71,411.41
XS GIS Cut Line= 6
 6420634.2406626 2050519.9369841 6420486.2598702 2051058.0488831
 6420176.8455508 2051703.7831334 6420008.6855854 2051979.5654975
 6419739.6296596 2052322.6118195 6419490.7529069 2052598.3941363
#Sta/Elev= 30
       0   84.12  343.26   83.84  394.41   65.84   405.3   64.03  445.81   66.97
  480.71   69.84  530.51   59.84   594.2   56.84  625.94   43.84  646.19   42.82
  671.04   35.87  765.09   33.53  783.54   36.62  798.74   42.86  828.47   43.84
  840.67   53.84  858.71   57.59  876.68   59.84  939.86   60.25 1861.47   59.51
 2203.31   60.99 2259.95   61.84 2276.08   63.84 2292.52   69.84 2314.85   70.51
  2345.9   73.84  2353.4    76.9 2370.43   83.84  2378.3   85.67 2404.61   87.77
#Mann= 3 ,-1 , 0
       0     .06       0  445.81    .035       0  2353.4     .05       0
Bank Sta=594.2,858.71
XS Rating Curve= 0 ,0
Exp/Cntr=0.3,0.1
