HEC-RAS study Baxter.prj: Baxter River GIS Example

--- Baxter.g02 (geometry) --- (continued)

Type RM Length L Ch R = 1 ,46534.  ,45.43,52.85,56.5
XS GIS Cut Line= 6
 6420177.1145989 2050176.0834706 6420082.9450296 2050586.3937977
  6419847.521059 2051467.5520186  6419705.997657 2052053.5558464
 6419564.7432558  2052497.498176 6419484.0265159 2052591.6677453
#Sta/Elev= 30
       0   83.45  637.64   79.84  676.06   77.84  723.04   63.84   735.6   63.84
  754.61   59.84  815.79    61.2  821.32   61.84  829.02   59.84  840.98   55.84
  848.43   51.25  857.27   43.84  871.81   42.43  873.72   40.92  899.55   35.24
  937.89    34.9  956.43   32.13  997.52   30.21 1007.45   30.51 1018.07   36.32
 1059.53   43.84 1079.29   53.84 1082.58   54.25 1172.73   59.84  1951.7   58.86
 2385.03   61.43 2475.45   73.84 2486.01   78.38 2503.37   85.08 2525.86   86.68
#Mann= 3 ,-1 , 0
       0     .05       0  815.79    .035       0 2486.01     .06       0
Bank Sta=848.43,1082.58
XS Rating Curve= 0 ,0
Exp/Cntr=0.3,0.1

Type RM Length L Ch R = 1 ,46481.  ,322.97,300.51,288.13
XS GIS Cut Line= 6
 6420109.5815457 2050230.7018379 6419941.4215803 2050963.8793138
 6419813.6200084 2051354.0104204 6419712.7240481 2051824.8583142
 6419544.8331307 2052476.5118113 6419450.6635614 2052604.3133832
#Sta/Elev= 30
       0   82.81  579.62   79.84  601.48   77.84  640.38   70.51   667.4   59.84
  737.51   59.84  747.11   60.95  755.38   61.84  762.91   59.84  776.99   53.84
  787.08   44.51  806.59    42.4  814.62    36.1  824.66    34.9  871.34    34.9
  890.75   31.89  931.35   29.81  941.34   30.16  952.85    36.3  994.29   43.84
 1021.34   53.59 1046.56   56.62 1109.28   59.84 1859.92   58.67 2304.04   60.56
    2342   63.84  2409.2   73.84 2425.14   82.29 2428.61   83.92 2475.96   87.13
#Mann= 3 ,-1 , 0
       0     .06       0  747.11    .035       0 2425.14     .05       0
Bank Sta=787.08,1021.34
XS Rating Curve= 0 ,0
Exp/Cntr=0.3,0.1

Type RM Length L Ch R = 1 ,46180.  ,272.51,260.8,234.04
XS GIS Cut Line= 4
  6419788.396042 2050047.4074926 6419594.9166842  2051078.469319
 6419263.6276303  2052327.902325 6419157.7961715 2052670.7029347
#Sta/Elev= 30
       0    81.2  521.74   79.84  593.11   77.84   671.5   77.78  719.36   75.84
  909.12   75.84  929.14   73.84  957.99   63.84  960.33   61.79   980.5   43.84
  993.16   34.32 1015.99   33.95 1030.33   32.03 1069.34   29.99 1080.89   34.85
 1094.53    38.1 1145.98   53.84 1160.22   55.27  1242.4   59.84 1408.12   59.84
 1468.29   57.84 1948.09   58.57 2218.38   57.84 2468.27   60.02  2493.2   63.43
 2528.53   76.12 2553.42   83.84 2634.34   87.84 2647.54   89.84 2700.43   89.84
#Mann= 3 ,-1 , 0
       0     .05       0  909.12    .035       0 2468.27     .06       0
Bank Sta=960.33,1160.22
XS Rating Curve= 0 ,0
Exp/Cntr=0.3,0.1

Type RM Length L Ch R = 1 ,45920.  ,250.93,280.31,313.43
XS GIS Cut Line= 5
 6419721.1320369 2049929.6955073 6419410.0361197 2050560.2953777
 6419309.1401121 2051224.5272508  6419183.020138 2051779.4551273
 6418871.9242208 2052477.3189555
#Sta/Elev= 30
       0   79.84  258.04   79.84  405.42   75.84   507.7   79.84  524.26   75.84
  563.85   73.84  910.28   71.58  964.15   71.84   983.5   79.84 1001.95   79.84
 1014.85   79.03 1038.18   71.84 1073.94   69.84 1087.53   67.84 1091.28   63.34
 1127.02   43.84 1131.69   33.03 1208.51   30.07 1239.39      43 1259.61   43.84
 1279.91   53.84 1298.97   55.84 1461.41    59.4 2358.49   60.13 2448.39   63.05
 2512.62   63.84 2553.71   76.55 2599.58   83.84 2650.59   87.84 2708.16   87.84
#Mann= 3 ,-1 , 0
       0     .06       0 1073.94    .035       0 2448.39     .05       0
#XS Ineff= 1 ,-1
       0  959.21   79.84
Permanent Ineff=
       F
Bank Sta=1091.28,1298.97
XS Rating Curve= 0 ,0
Exp/Cntr=0.3,0.1

Type RM Length L Ch R = 1 ,45639.  ,229.21,228.25,215.91
XS GIS Cut Line= 6
 6419729.5400257 2049702.6795729 6419359.5881396 2050165.1194779
 6419098.9401552 2050778.9033234 6419040.0841863 2051115.2232543
  6418863.516232 2051569.2551705 6418678.5402889 2052536.1749718
#Sta/Elev= 30
       0   79.84  301.97   79.84  431.23   79.69   543.9   77.84  580.83   75.84
   782.5   72.48 1016.53   71.84  1203.7   69.84 1273.48   67.84 1338.61   67.84
 1360.94   63.13 1399.43   43.84 1408.89   34.02 1422.21   34.47 1477.81   31.72
 1503.48    37.4  1516.9   42.33 1537.07   43.84 1560.54   53.84 1590.89   54.56
 1724.03   57.34 1906.83   57.23 2053.42   60.49 2591.92   63.84  2607.2   63.84
 2658.93   73.84 2725.41   83.84 2766.29   85.84 2785.05   87.84 3072.09   87.84
#Mann= 4 ,-1 , 0
       0     .05       0  301.97     .06       0 1338.61    .035       0
 2591.92     .05       0
#XS Ineff= 1 ,-1
       0 1292.18   79.84
Permanent Ineff=
       F
Bank Sta=1360.94,1590.89
XS Rating Curve= 0 ,0
Exp/Cntr=0.3,0.1

Type RM Length L Ch R = 1 ,45411.  ,111.19,121.08,110.37
XS GIS Cut Line= 6
 6419670.6398938 2048731.0497263 6419168.9735946  2049743.847714
 6419047.0796254 2050108.8195129 6418778.0236996 2051178.3168723
  6418542.599729 2052126.7390983 6418455.1565508 2052510.1438139
#Sta/Elev= 30
       0      83  236.64   81.84  496.12    76.8   681.3   76.17 1220.72   79.84
 1272.56   76.56 1420.03   71.84 1554.57   73.47  2123.4   73.09 2173.97   69.83
 2224.13   63.84 2241.54   53.84 2248.73   51.08 2276.11   39.65 2288.58    38.4
 2302.14      32 2313.56   33.64 2327.94   31.76  2396.2      35 2416.41   37.73
 2478.35   53.84 2510.43   55.04 2890.56   56.48 3162.29    63.1 3380.07   63.84
 3391.05   63.84 3447.18   73.23 3480.91   80.87 3516.95   83.84  3988.3   87.32
#Mann= 3 ,-1 , 0
       0     .06       0 2241.54    .035       0 3380.07     .06       0
#XS Ineff= 2 ,-1
       0    2170    80.5    3420    3500      85
Permanent Ineff=
       F       F
Bank Sta=2248.73,2510.43
XS Rating Curve= 0 ,0
Exp/Cntr=0.3,0.1

Type RM Length L Ch R = 3 ,45360.  ,,,
Node Name=Railroad
Bridge Culvert--1,0,-1,-1, 0
Deck Dist Width WeirC Skew NumUp NumDn MinLoCord MaxHiCord MaxSubmerge Is_Ogee
40,20,2.6,0, 136, 136, , , 0.95, 0, 0,0,,
       0    4.85   14.53   17.81   27.63   31.57   42.17   51.18   57.44   64.66
   71.66   79.77   86.38  104.19  119.01  124.35  138.85  144.88  159.58  164.55
  170.18   196.4  199.96   224.4  226.64  244.51  246.31  251.49  253.74  273.43
  290.48  304.22  310.25  333.81  334.66  335.96  365.36  365.66  373.82  423.93
  424.73  426.85   452.9  455.21  460.12  472.74  478.41  484.98  490.53  493.89
  497.85  502.85  521.82  524.66  532.35  561.74  570.35  579.03  608.33  615.57
  641.11  647.87   676.5  681.04  709.17  711.85  746.87  747.13  750.93  781.25
  782.67  803.96  805.36  822.43  824.29  842.86  846.32  849.93  867.05  872.15
  886.31  892.52  896.67  903.35   916.3  923.76  932.93  941.83  955.05  964.87
  975.94   985.5  997.46 1002.64 1015.62  1030.3 1036.52 1051.63 1053.66 1069.81
 1071.42 1080.93 1092.16 1105.41 1118.24  1128.8 1141.64  1145.1 1151.45 1161.03
 1162.72 1166.28 1173.24 1181.95 1185.49 1194.24  1195.5 1203.25 1204.61 1204.72
 1213.27 1221.36 1222.49 1230.49 1238.01 1240.35 1246.39 1248.23 1251.92 1269.91
 1276.11    2200    2200    3400    3400    3900
   83.84   83.84   83.84   83.84   83.84   83.84   83.84   83.84   83.84   83.84
   83.84   83.84   83.84   83.84   83.84   83.84   83.84   83.84   83.84   83.84
   83.84   83.84   83.84   83.84   83.84   83.84   83.81   83.74   83.68   83.35
   83.06   82.65   82.34   82.15   82.03   81.84   81.84   81.84   81.84   81.69
   81.67   81.56   81.42   81.12      81   80.88   80.72   80.53   80.47   80.36
   80.23   80.19   80.26   80.24   80.23   80.05   80.04   80.03   80.33   80.33
   80.61    80.7   81.01   81.07   81.37   81.41    81.8    81.8   81.84   81.84
   81.84   81.84   81.84   81.84   81.84   81.84   81.84   81.84   81.84   81.84
   81.84   81.84   81.84   81.84   81.84   81.84   81.84   81.84   81.84   81.84
   81.84   81.84   81.84   81.84   81.84   81.84   81.84   81.84   81.84   81.84
   81.84   81.84   81.48   81.05   80.77   80.39   79.84   79.69   79.41   79.49
   79.36    79.1   79.24   79.41   79.51   79.67   79.71   79.84   79.85   79.85
   79.91   79.96   79.98   80.04   80.09   80.14   79.79   79.88   79.81   80.15
   80.29      81      82      85      85      86
                                                                                
                                                                                
                                                                                
                                                                                
                                                                                
                                                                                
                                                                                
                                                                                
                                                                                
                                                                                
                                                                                
                                                                                
                                                                                
               0      74      78       0       0
       0    4.85   14.53   17.81   27.63   31.57   42.17   51.18   57.44   64.66
   71.66   79.77   86.38  104.19  119.01  124.35  138.85  144.88  159.58  164.55
  170.18   196.4  199.96   224.4  226.64  244.51  246.31  251.49  253.74  273.43
  290.48  304.22  310.25  333.81  334.66  335.96  365.36  365.66  373.82  423.93
  424.73  426.85   452.9  455.21  460.12  472.74  478.41  484.98  490.53  493.89
  497.85  502.85  521.82  524.66  532.35  561.74  570.35  579.03  608.33  615.57
  641.11  647.87   676.5  681.04  709.17  711.85  746.87  747.13  750.93  781.25
  782.67  803.96  805.36  822.43  824.29  842.86  846.32  849.93  867.05  872.15
  886.31  892.52  896.67  903.35   916.3  923.76  932.93  941.83  955.05  964.87
  975.94   985.5  997.46 1002.64 1015.62  1030.3 1036.52 1051.63 1053.66 1069.81
 1071.42 1080.93 1092.16 1105.41 1118.24  1128.8 1141.64  1145.1 1151.45 1161.03
 1162.72 1166.28 1173.24 1181.95 1185.49 1194.24  1195.5 1203.25 1204.61 1204.72
 1213.27 1221.36 1222.49 1230.49 1238.01 1240.35 1246.39 1248.23 1251.92 1269.91
 1276.11    2200    2200    3400    3400    3900
   83.84   83.84   83.84   83.84   83.84   83.84   83.84   83.84   83.84   83.84
   83.84   83.84   83.84   83.84   83.84   83.84   83.84   83.84   83.84   83.84
   83.84   83.84   83.84   83.84   83.84   83.84   83.81   83.74   83.68   83.35
   83.06   82.65   82.34   82.15   82.03   81.84   81.84   81.84   81.84   81.69
   81.67   81.56   81.42   81.12      81   80.88   80.72   80.53   80.47   80.36
   80.23   80.19   80.26   80.24   80.23   80.05   80.04   80.03   80.33   80.33
   80.61    80.7   81.01   81.07   81.37   81.41    81.8    81.8   81.84   81.84
   81.84   81.84   81.84   81.84   81.84   81.84   81.84   81.84   81.84   81.84
   81.84   81.84   81.84   81.84   81.84   81.84   81.84   81.84   81.84   81.84
   81.84   81.84   81.84   81.84   81.84   81.84   81.84   81.84   81.84   81.84
   81.84   81.84   81.48   81.05   80.77   80.39   79.84   79.69   79.41   79.49
   79.36    79.1   79.24   79.41   79.51   79.67   79.71   79.84   79.85   79.85
   79.91   79.96   79.98   80.04   80.09   80.14   79.79   79.88   79.81   80.15
   80.29      81      82      85      85      86
                                                                                
                                                                                
                                                                                
                                                                                
                                                                                
                                                                                
                                                                                
                                                                                
                                                                                
                                                                                
                                                                                
                                                                                
                                                                                
               0      74      78       0       0
Pier Skew, UpSta & Num, DnSta & Num=  ,2250, 2 ,2250, 2 , 0 , 0 , 0 ,,
      10      10
   29.12      78
      10      10
   29.12      78
Pier Skew, UpSta & Num, DnSta & Num=  ,2350, 2 ,2350, 2 , 0 , 0 , 0 ,,
      10      10
   29.12      78
      10      10
   29.12      78
Pier Skew, UpSta & Num, DnSta & Num=  ,2450, 2 ,2450, 2 , 0 , 0 , 0 ,,
      10      10
   29.12      78
      10      10
   29.12      78
Pier Skew, UpSta & Num, DnSta & Num=  ,2550, 2 ,2550, 2 , 0 , 0 , 0 ,,
      10      10
   29.12      78
      10      10
   29.12      78
Pier Skew, UpSta & Num, DnSta & Num=  ,2650, 2 ,2650, 2 , 0 , 0 , 0 ,,
      10      10
   29.12      78
      10      10
   29.12      78
Pier Skew, UpSta & Num, DnSta & Num=  ,2750, 2 ,2750, 2 , 0 , 0 , 0 ,,
      10      10
   29.12      78
      10      10
   29.12      78
Pier Skew, UpSta & Num, DnSta & Num=  ,2850, 2 ,2850, 2 , 0 , 0 , 0 ,,
      10      10
   29.12      78
      10      10
   29.12      78
Pier Skew, UpSta & Num, DnSta & Num=  ,2950, 2 ,2950, 2 , 0 , 0 , 0 ,,
      10      10
   29.12      78
      10      10
   29.12      78
Pier Skew, UpSta & Num, DnSta & Num=  ,3050, 2 ,3050, 2 , 0 , 0 , 0 ,,
      10      10
   29.12      78
      10      10
   29.12      78
Pier Skew, UpSta & Num, DnSta & Num=  ,3150, 2 ,3150, 2 , 0 , 0 , 0 ,,
      10      10
   29.12      78
      10      10
   29.12      78
Pier Skew, UpSta & Num, DnSta & Num=  ,3250, 2 ,3250, 2 , 0 , 0 , 0 ,,
      10      10
   29.12      78
      10      10
   29.12      78
Pier Skew, UpSta & Num, DnSta & Num=  ,3350, 2 ,3350, 2 , 0 , 0 , 0 ,,
      10      10
   29.12      78
      10      10
   29.12      78
BR Coef=-1 , 0 , 0 ,, 0 ,,,0.8,0,,0,
WSPro=,,,, 1 ,,,, 0 ,,,, 0 ,,,,-1 ,-1 ,-1 , 0 , 0 , 0 , 0 , 0
BC Design=,, 0 ,, 0 ,,12,2250,2250,100,10
BC HTab HWMax=95
BC HTab MaxFlow=200000
BC Use User HTab Curves=0
BC User HTab FreeFlow(D)= 0

Type RM Length L Ch R = 1 ,45290.  ,274.1,256.23,255.57
XS GIS Cut Line= 5
 6419578.4651333  2048682.823002 6419080.7116279 2049651.4244011
 6418724.0997263 2050898.6266844 6418448.4301597 2052167.0974919
  6418394.618984  2052321.804628
#Sta/Elev= 30
       0   79.84 1089.01   76.08 1156.34   77.84 1286.91   75.84 1348.02   71.84
 2109.82   73.32 2146.65   63.84  2183.2   63.84 2255.88   53.84 2276.17   45.59
 2289.32    37.3 2299.36    34.2 2309.38    37.3 2324.41    30.7 2364.53   29.12
 2449.58    39.8 2454.58    37.6 2474.58    37.2 2534.14   43.84  2545.5   53.84
 2550.79   54.28 2568.29   55.84 2965.46    56.1 3216.19   61.27 3238.34   63.84
 3362.69   63.84 3398.55   69.32 3423.05   78.44 3469.73   83.84 3848.07   85.07
#Mann= 3 ,-1 , 0
       0     .06       0  2183.2    .035       0 3362.69     .06       0
#XS Ineff= 2 ,-1
       0    2180      79    3420    3500      79
Permanent Ineff=
       F       F
Bank Sta=2276.17,2550.79
XS Rating Curve= 0 ,0
Exp/Cntr=0.3,0.1

Type RM Length L Ch R = 1 ,45034.  ,282.79,257.86,241.35
XS GIS Cut Line= 5
 6419559.9675579 2048427.2198583 6418919.2780535 2049637.9716191
 6418487.4647081 2050661.9916188 6418459.0684926 2051002.7461094
 6418165.9214518 2051850.9567342
#Sta/Elev= 30
       0   79.93   969.5   75.84 1286.17   77.84 1498.23   75.84 1553.07   71.84
 2046.48   71.84 2492.63   65.84  2550.5   57.54 2566.92   55.48    2599   43.84
 2608.83   38.04  2619.4   35.73 2632.17   38.02    2648   30.92 2657.21      32
 2666.65   30.25 2690.82   29.81 2738.85   37.44 2767.05   37.82 2784.18   43.84
 2812.88   48.41 2828.98   53.84 2843.64   54.26 2960.33   55.84 3468.07   55.84
 3517.02   55.84 3536.07   63.84 3575.45   73.84 3589.23   83.84 3720.54   85.84
#Mann= 3 ,-1 , 0
       0     .06       0 2492.63    .035       0 3468.07     .05       0
#XS Ineff= 2 ,-1
       0 2337.5379.93319 3512.78 3720.54   85.84
Permanent Ineff=
       F       F
Bank Sta=2550.5,2843.64
XS Rating Curve= 0 ,0
Exp/Cntr=0.3,0.1

Type RM Length L Ch R = 1 ,44776.  ,335.08,331.39,355.75
XS GIS Cut Line= 6
 6419492.7035528 2048032.0439584 6419013.4476701 2048544.9318436
 6418651.9037255 2049276.4276744 6418279.5685582 2050420.8633937
 6418147.4238291 2051260.7152573 6417920.4078947 2051840.8671476
#Sta/Elev= 30
       0      80   511.9   76.06  574.06   56.25  648.81   53.84  704.26   53.84
 1090.47   77.43  1360.2   77.84 1475.49   73.84 1852.28   69.45 2200.47    70.2
 2815.83   66.25 2862.07   65.84 2897.83   61.63 2942.31   57.34 2970.68   55.84
  3025.1   43.84 3084.01   37.55 3093.49   38.38 3106.96   30.28 3116.21      32
  3162.9      31 3197.25   34.19 3215.93   38.67 3259.04   53.84 3282.24   53.97
 3717.74   55.84 3773.75   72.78 3893.12   83.84 3986.27   85.84 4194.57   85.84
#Mann= 3 ,-1 , 0
       0     .06       0 2897.83    .035       0 3773.75     .06       0
#XS Ineff= 2 ,-1
       0 2713.19      80 3733.94 4194.57   85.84
Permanent Ineff=
       F       F
Bank Sta=2942.31,3282.24
XS Rating Curve= 0 ,0
Exp/Cntr=0.3,0.1

Type RM Length L Ch R = 1 ,44444.  ,191.29,187.6,190.02
XS GIS Cut Line= 6
 6419557.0550794 2047642.5285289  6418744.391697 2048191.7959351
 6418525.3263129 2048428.1568878 6418265.1358144 2048948.5157323
 6418046.5278688 2049747.2755682 6417718.6159267 2051916.5391415
#Sta/Elev= 30
       0   80.11  204.65   71.78  319.73      75  434.03      65  748.38   55.84
  766.43   55.84   835.7   75.15 1012.49   79.84 2523.31   64.49 2716.12   75.54
 3203.58   75.05 3259.91   72.84 3282.83   63.84 3329.68   57.84 3429.03   53.77
 3470.57   43.84 3568.94   42.26 3625.99    46.4 3700.55   39.15 3712.25   33.84
 3773.14   31.29 3793.21   32.73 3817.45   43.84 3873.88   54.93 3976.44    76.5
 4141.73   80.32 4202.48   68.07 4286.28   63.84 4327.64   83.84 4910.04   85.84
#Mann= 3 ,-1 , 0
       0     .06       0 3203.58    .035       0 4202.48     .06       0
#XS Ineff= 2 ,-1
       0    3220      74    3960 4908.64   85.84
Permanent Ineff=
       F       F
Bank Sta=3429.03,3873.88
XS Rating Curve= 0 ,0
Exp/Cntr=0.3,0.1

Type RM Length L Ch R = 3 ,44367.  ,,,
Node Name=Highway
Bridge Culvert--1,0,-1,-1, 0
Deck Dist Width WeirC Skew NumUp NumDn MinLoCord MaxHiCord MaxSubmerge Is_Ogee
40,90,2.6,0, 7, 7, , , 0.95, 0, 0,0,,
    1500    3000    3250    3250    3900    3900    5000
      70      75      81      81      86      86      87
                              74      74
    1500    3000    3300    3300    4000    4000    5000
      70      75      81      81      86      86      87
                              74      74
Pier Skew, UpSta & Num, DnSta & Num=  ,3300, 2 ,3340, 2 , 0 , 0 , 0 ,,
       4       4
   31.29      74
       4       4
   31.29      74
Pier Skew, UpSta & Num, DnSta & Num=  ,3395, 2 ,3435, 2 , 0 , 0 , 0 ,,
       4       4
   31.29      74
       4       4
   31.29      74
Pier Skew, UpSta & Num, DnSta & Num=  ,3490, 2 ,3530, 2 , 0 , 0 , 0 ,,
       4       4
   31.29      74
       4       4
   31.29      74
Pier Skew, UpSta & Num, DnSta & Num=  ,3585, 2 ,3625, 2 , 0 , 0 , 0 ,,
       4       4
   31.29      74
       4       4
   31.29      74
Pier Skew, UpSta & Num, DnSta & Num=  ,3680, 2 ,3720, 2 , 0 , 0 , 0 ,,
       4       4
   31.29      74
       4       4
   31.29      74
Pier Skew, UpSta & Num, DnSta & Num=  ,3775, 2 ,3815, 2 , 0 , 0 , 0 ,,
       4       4
   31.29      74
       4       4
   31.29      74
Pier Skew, UpSta & Num, DnSta & Num=  ,3870, 2 ,3910, 2 , 0 , 0 , 0 ,,
       4       4
   31.29      74
       4       4
   31.29      74
BR Coef=-1 , 0 , 0 ,, 0 ,,,0.8,0,,0,
WSPro=,,,, 1 ,,,, 0 ,,,, 0 ,,,,-1 ,-1 ,-1 , 0 , 0 , 0 , 0 , 0
BC Design=,, 0 ,, 0 ,,7,3300,3340,95,4
BC HTab HWMax=95
BC HTab MaxFlow=200000
BC Use User HTab Curves=0
BC User HTab FreeFlow(D)= 0

Type RM Length L Ch R = 1 ,44257.  ,119.44,428.14,566.78
XS GIS Cut Line= 6
 6419274.0956071 2047477.1160819 6418834.7329641 2047738.3947009
 6418349.2157971 2048200.2039239 6418029.7118438 2048906.4757409
 6417802.6959094 2050075.1875103 6417567.2719388 2051815.6431338
#Sta/Elev= 30
       0      80  229.64      75  655.66   77.84  695.03    81.7  768.38      77
  800.43   81.84 1118.44    66.6 1533.08   69.99 1557.11   65.54 1791.89   67.87
 2780.24   59.84 3171.67   61.79 3293.47   62.17 3424.79   51.03 3456.03   43.84
  3555.2   42.26 3617.95    46.4 3801.71    31.5 3826.52    32.6 3855.05   43.84
  3891.9   48.84 3933.55   53.84 4014.33   79.39 4146.06   83.14 4224.48   83.84
 4265.14   63.84 4352.99   63.84 4388.53   83.84 4832.35   83.84 4904.25   80.11
#Mann= 3 ,-1 , 0
       0     .06       0 3171.67    .035       0 4146.06     .05       0
#XS Ineff= 2 ,-1
       0    3280      70    4000 4904.25  80.109
Permanent Ineff=
       F       F
Bank Sta=3424.79,3891.9
XS Rating Curve= 0 ,0
Exp/Cntr=0.3,0.1

Type RM Length L Ch R = 1 ,43829.  ,414.85,442.62,553.77
XS GIS Cut Line= 6
 6419101.7316473  2047475.014061   6418260.93182 2048231.7339056
 6418061.2418729 2048694.1738106 6417693.3919129 2050207.6134997
 6417220.4420456 2050554.4433929 6416968.2020974  2050659.543395
#Sta/Elev= 30
       0      80  108.54   75.41  123.35   77.84  515.48   77.84  538.75   81.84
  592.47   81.84  606.99   79.92  639.79   81.84  750.93   73.84  837.85   70.87
 1391.42   71.84 1429.65   69.64 1764.35   65.64 2325.82   65.84 2928.65   58.47
 3302.98   57.84 3334.48   54.23 3386.99   43.84  3433.5   42.26 3469.99   45.95
 3552.93   36.12 3646.22    31.6 3661.97   35.25 3681.89   43.84 3728.17   47.01
 3811.36   52.68 3828.57   53.84 3864.81   63.84 3896.35   83.84 4054.22   85.84
#Mann= 3 ,-1 , 0
       0     .06       0 2928.65    .035       0 3811.36     .05       0
#XS Ineff= 1 ,-1
       0 3073.36      70
Permanent Ineff=
       F
Bank Sta=3334.48,3728.17
XS Rating Curve= 0 ,0
Exp/Cntr=0.3,0.1

Type RM Length L Ch R = 1 ,43386.  ,462.42,634.69,621.98
XS GIS Cut Line= 6
 6419028.1616269 2047443.4840793 6418239.9118007 2048147.6539228
 6417766.9619333 2049524.4636282 6417535.7419571 2049850.2735494
   6417336.05201 2050028.9435245  6416894.632077 2050060.4735062
#Sta/Elev= 30
       0   78.01  414.74   78.25  473.23   81.84  524.92   81.84  621.09   77.84
  688.73   71.84 1405.14   71.84 1773.03   65.38    2159   65.84 2385.14   61.75
  2750.2   57.65 2825.95   55.84 2936.09   49.84 3024.69   49.84 3048.46   55.84
 3169.64   57.84 3184.06   53.84 3194.76    48.7 3206.24   43.84 3212.62   37.63
 3242.01      38 3249.85    35.8 3302.87    32.5  3314.2      37 3340.03   43.04
  3377.4   53.84 3419.95   73.84 3430.44   83.84 3451.88   83.94 3625.61   84.84
#Mann= 3 ,-1 , 0
       0     .06       0 2385.14    .035       0 3451.88     .05       0
#XS Ineff= 1 ,-1
   37.42 2743.48      68
Permanent Ineff=
       F
Bank Sta=3194.76,3340.03
XS Rating Curve= 0 ,0
Exp/Cntr=0.3,0.1

Type RM Length L Ch R = 1 ,42751.  ,688.21,642.75,621.09
XS GIS Cut Line= 6
  6418744.391697 2047517.0540524 6418102.2664965 2048230.6398683
 6417777.4718957 2049209.1637166 6417493.7019658 2049398.3436541
 6417190.7047079 2049403.0932234 6416663.4121482 2049555.9936099
#Sta/Elev= 30
       0   77.84  158.46   79.84  319.42   75.84  535.09   74.98  551.55   73.84
  710.17   71.84 1230.07   71.33 1571.26   64.95 1816.74    64.9 1941.13   63.84
 2036.78   55.84 2298.77   55.84 2343.69    54.3 2398.43   45.84 2408.96   42.33
  2427.9   34.62 2472.18   36.58 2477.97    34.6 2527.27      32  2551.5    39.8
 2573.71   43.84 2601.59   46.83 2630.43   49.92 2652.72   53.84 2686.81   63.84
 2705.01   73.84 2719.29   75.84 2793.73   75.84  2901.3    82.1 3184.08   85.74
#Mann= 3 ,-1 , 0
       0     .06       0 1816.74    .035       0  2901.3     .05       0
#XS Ineff= 1 ,-1
       0 2262.99      68
Permanent Ineff=
       F
Bank Sta=2408.96,2601.59
XS Rating Curve= 0 ,0
Exp/Cntr=0.3,0.1

Type RM Length L Ch R = 1 ,42109.  ,377.39,372.57,283.73
XS GIS Cut Line= 6
 6418644.9204513 2047539.3136146 6417968.4614228 2048319.8432665
 6417492.7100285 2048743.5593254 6417121.0292104 2048788.1610482
 6416950.0560738 2048914.5325093 6416712.1803766 2049107.8064837
#Sta/Elev= 30
       0   77.84  218.66   75.84  475.47   75.84  491.66   73.84  661.11   71.84
 1145.17   69.84 1298.19   69.84    1503   63.84    1529   55.84 1682.18   53.84
 1701.27   51.33 1731.97   49.84  1740.4   48.24 1758.81   43.84 1763.15    32.9
 1797.26    34.7 1876.22    31.5 1885.06   35.54 1931.17    44.9 2015.23   55.84
 2061.12   57.41 2097.39   61.64 2128.42   73.84 2161.39   77.84 2324.26   75.84
  2376.9   78.07 2416.94   78.18 2443.89   78.24 2528.25   81.84  2563.4   81.84
#Mann= 3 ,-1 , 0
       0     .06       0 1145.17    .035       0 2416.94     .05       0
Bank Sta=1740.4,1931.17
XS Rating Curve= 0 ,0
Exp/Cntr=0.3,0.1

Type RM Length L Ch R = 1 ,41736.  ,287.7,367.05,432.26
XS GIS Cut Line= 6
 6418660.3117143   2047422.46406 6418166.3418276 2047821.8440016
 6417916.4260874   2048141.43647 6417492.7100285 2048327.2768791
  6417039.259472  2048527.984466 6416652.7114287 2048929.3997345
#Sta/Elev= 30
       0   76.84   76.91   77.36  128.07   75.84  617.34   75.84  660.06   73.84
  1053.9   70.73 1224.79   69.84 1311.19   67.84 1333.25   63.84 1358.61   53.84
  1363.4   53.28 1379.98   52.25 1474.92   51.37 1544.41   48.38 1569.29   46.09
 1584.85   43.84 1618.61    33.6 1733.36    31.6 1782.62   43.84 1811.24    47.9
 1854.23   53.84 2046.02   55.84 2176.11   55.84 2241.57   57.84 2306.77   63.74
 2379.89   74.28 2388.59   77.84 2394.49   75.84 2404.24   81.84 2556.77   81.84
#Mann= 3 ,-1 , 0
       0     .06       0  1053.9    .035       0 2379.89     .05       0
Bank Sta=1569.29,1811.24
XS Rating Curve= 0 ,0
Exp/Cntr=0.3,0.1

Type RM Length L Ch R = 1 ,41369.  ,425.26,426.3,407.56
XS GIS Cut Line= 6
 6418534.1917402 2047369.9141063 6418113.7918266 2047790.3140199
 6417535.7419571 2048011.0239391 6417125.8520532 2048032.0439584
 6416863.1020953 2048147.6539228  6416358.622199 2048504.9938258
#Sta/Elev= 30
       0   75.84     495   75.84   536.9   73.84  793.95   72.33  905.69   71.84
 1111.02   67.84 1171.12   63.84 1207.39   53.84 1213.27   51.84 1219.68   47.84
 1242.79   46.51 1264.13   46.82  1323.5   49.84 1335.74   47.94 1351.06   45.84
 1356.33    44.2 1380.14    33.6 1480.71    31.6 1549.43   45.11  1615.5   55.84
 2191.38   57.84 2249.83   60.88 2295.26   63.84 2324.67   68.35 2358.28   71.84
 2383.23   75.84 2387.86   77.84 2467.55   79.84 2496.43   81.84 2528.99   81.85
#Mann= 3 ,-1 , 0
       0     .06       0  793.95    .035       0 2249.83     .06       0
Bank Sta=1335.74,1549.43
XS Rating Curve= 0 ,0
Exp/Cntr=0.3,0.1

Type RM Length L Ch R = 1 ,40943.  ,826.24,806.49,525.17
XS GIS Cut Line= 5
 6418544.7017499 2047075.6341667 6417840.5319064 2047485.5240707
 6417451.6619744 2047601.1340351 6417094.3220715 2047590.6240254
 6416011.7923057 2048200.2039239
#Sta/Elev= 30
       0   76.22  639.15   75.84  656.33   73.84 1134.23   69.84  1217.7   67.84
 1220.96   65.84 1232.53   63.84 1252.65   53.84 1273.64   48.64 1292.99   43.84
 1302.66    33.6 1317.89    32.1 1368.19   31.66 1382.38    35.4 1447.09   43.69
 1461.05   45.84    1482   51.84  1514.5   53.84 1630.27   55.84 1666.52   59.84
 1852.17   57.49 2429.48   60.79 2491.93   64.07 2518.97   67.84 2520.22   69.84
 2540.59   73.84 2632.38   79.37 2700.12   79.84 2720.74   81.84 2820.33   81.84
#Mann= 3 ,-1 , 0
       0     .06       0  1217.7    .035       0 2429.48     .06       0
Levee=0,,,-1,2630.25,79.95625,,	380
Bank Sta=1273.64,1447.09
XS Rating Curve= 0 ,0
Exp/Cntr=0.3,0.1

Type RM Length L Ch R = 1 ,40136.  ,661.44,655.91,599.95
XS GIS Cut Line= 4
 6417903.5918697 2046592.1742424  6417484.132157 2046781.1770076
 6417190.7047079 2046932.6234269 6415759.5523575 2047800.8239823
#Sta/Elev= 30
       0   75.87  236.55   76.59  294.15   75.84  430.11   69.84  442.09   67.84
  454.69   63.84  462.37   53.84  475.83   43.01  505.14    29.1  576.25    31.5
  584.74    32.4  622.26   43.84  636.05   45.84  736.07    47.5  753.33   47.84
  802.34   53.84 1076.03   55.84 1213.27   57.84 2022.79   57.84 2026.26   60.17
 2041.79   61.84 2050.26   63.84 2052.71   67.84  2089.1   73.84 2096.25   74.32
 2182.76   79.84 2242.23   80.47  2297.4   79.95 2360.19   81.84 2464.19   81.84
#Mann= 2 ,-1 , 0
       0    .035       0 2096.25     .05       0
Levee=0,,,-1,2197.8,80.22,,	380
Bank Sta=475.83,736.07
XS Rating Curve= 0 ,0
Exp/Cntr=0.3,0.1

Type RM Length L Ch R = 1 ,39480.  ,474.01,468.09,436.4
XS GIS Cut Line= 3
 6417893.0819074 2045709.3344237 6415781.0439683 2047160.8173223
 6415330.6130551 2047856.6583672
#Sta/Elev= 30
       0   75.66   96.61   73.84  379.71   73.84  561.59   77.84  654.78   77.84
  900.46   71.84  923.73   63.84  931.22   53.84  941.88   45.31   943.7   43.84
  966.28   38.92  977.12   34.62 1003.42   30.02 1015.09    29.5  1040.2   31.68
 1084.75    32.6 1130.21   45.51 1207.42   53.61 1348.98   55.84  1676.3   55.84
 1965.59   58.93 2238.46   57.84 2270.31   59.71 2349.15   57.44  2449.3   57.84
 2580.91   66.44 2611.63   67.84 2702.79   75.84 3084.13   79.84 3391.62   80.13
#Mann= 3 ,-1 , 0
       0     .06       0  561.59    .035       0 2580.91     .06       0
Levee=0,,,-1,2661.54,77.33,,	380
Bank Sta=941.88,1130.21
XS Rating Curve= 0 ,0
Exp/Cntr=0.3,0.1

Type RM Length L Ch R = 1 ,39012.  ,742.69,700.15,609.51
XS GIS Cut Line= 5
 6417399.1119734 2045520.1544863 6416810.5521416 2045877.4943892
 6416631.8821665 2046024.6343826 6415512.0072129 2046872.3175141
 6414847.1531781  2048014.308323
#Sta/Elev= 30
       0   73.84  254.94   75.84  314.61   77.84  449.27   77.84  624.32   73.84
     640   63.84  666.56   56.33  690.09   47.81  701.08   43.84  721.17    39.2
  772.72   29.61  798.12      32  848.65    32.6  861.46    35.7  872.52   43.84
  877.88   46.27  894.55   53.84  904.32   55.84  942.79   58.17 1064.65   58.71
 1327.75   56.78 1736.01   57.84 1756.62   55.84 1910.57   55.84 1978.27   57.15
 2191.68   55.84 2229.53   57.84 2285.94   63.78 2369.72   75.84 3645.96   79.84
#Mann= 3 ,-1 , 0
       0     .06       0  314.61    .035       0 2285.94     .06       0
Levee=0,,,-1,2364.84,75.81,,	380
Bank Sta=690.09,877.88
XS Rating Curve= 0 ,0
Exp/Cntr=0.3,0.1

Type RM Length L Ch R = 1 ,38312.  ,374.38,367.97,323.69
XS GIS Cut Line= 4
  6416859.415654 2044585.2038341 6416064.3219057 2045673.7250315
 6415246.5330724 2046458.8286426 6414405.7332451 2047930.2283403
#Sta/Elev= 30
       0   85.65    7.24   85.79   41.85   83.84   70.01   85.84  276.11   85.84
   398.3   81.84  482.18   73.84     531   73.84  911.56   73.84 1015.52   63.84
 1035.88   48.65 1040.27   43.84 1080.99      37 1081.52    40.8 1101.68    32.3
 1113.67    31.9 1195.81    34.1 1208.17    44.1 1249.02   49.84 1548.48   55.84
 1660.85   61.84 1728.69   61.84 1798.53   57.84 2031.24   57.84 2335.57   53.84
 2407.72   53.84  2461.9   59.17 2530.41   75.84  3587.1   75.84 4176.32   79.98
#Mann= 4 ,-1 , 0
       0     .06       0    7.24     .06       0     531    .035       0
  2461.9     .06       0
Levee=0,,,-1,2527.47,76.67,,	380
Bank Sta=1035.88,1208.17
XS Rating Curve= 0 ,0
Exp/Cntr=0.3,0.1

Type RM Length L Ch R = 1 ,37944.  ,606.16,578.05,519.9
XS GIS Cut Line= 5
 6416434.1628402 2044461.9290764 6415971.7229352   2045166.09892
 6415751.0129688 2045502.4188509 6415057.3531349 2046301.1786868
 6414121.9633152 2048035.3283424
#Sta/Elev= 30
       0   85.84  244.26   83.84  285.92   79.84  332.83   79.84  369.94   73.84
  418.97   73.84   761.4   73.53  787.53   69.84  869.79   67.84  882.67   63.84
  898.95      51  911.77   43.84  968.36   39.47  992.51    32.8 1038.87   31.99
  1080.3    33.5 1093.83   43.84 1103.96   46.21 1144.27   51.84 1336.67   55.77
 1419.25   61.84 1525.21   57.84 2134.18   53.84 2193.73   53.84 2248.61   60.72
 2267.59   63.84 2296.83   73.84 2331.18   75.84 3137.03   74.65 4272.96   79.84
#Mann= 3 ,-1 , 0
       0     .06       0  418.97    .035       0 2248.61     .05       0
Levee=0,,,-1,2330.57,74.77473,,	380
Bank Sta=898.95,1103.96
XS Rating Curve= 0 ,0
Exp/Cntr=0.3,0.1

Type RM Length L Ch R = 1 ,37366.  ,589.97,558.31,507.96
XS GIS Cut Line= 5
 6415793.0529601 2044304.2791207 6415456.7330292 2044840.2889987
 6415278.0630541 2045229.1589307 6414678.9932126 2046059.4487483
  6413817.173366 2048003.7983133
#Sta/Elev= 30
       0   85.87  332.34   81.84  362.04   77.68  438.32   71.84  669.63   65.84
  686.69   63.84  704.62   49.32  713.45   43.84  717.84   43.66  806.15      40
  842.34    32.8  885.71      32  921.86    33.5  924.98   45.84  938.07   48.23
  976.46   51.84 1214.05   57.84 1452.13   57.84 1564.35   53.84 1793.01   53.84
 1849.03   57.45 1862.29   53.84 1903.78   53.84 1942.65   55.84 2066.85   69.84
  2130.9   73.84 2847.47   73.84  3394.2   69.64 3478.39   73.84 4211.37    80.1
#Mann= 3 ,-1 , 0
       0     .06       0  362.04    .035       0  2130.9     .05       0
Levee=0,,,-1,2202.75,74.34217,,	380
Bank Sta=717.84,938.07
XS Rating Curve= 0 ,0
Exp/Cntr=0.3,0.1

Type RM Length L Ch R = 1 ,36808.  ,564.92,652.32,662.06
XS GIS Cut Line= 6
 6415299.0830734 2043862.8591877 6415067.8630973 2044199.1791186
 6414857.6631404  2044756.209016 6414794.6031771 2045039.9789459
  6414258.593299 2045807.2088001 6413522.8934265   2047940.73835
#Sta/Elev= 30
       0    82.8  104.68   81.84  205.51   75.84  407.57   73.84  436.54   67.84
  630.47   66.35  1026.1   65.84 1031.08   63.84 1038.18   43.84 1051.62   42.71
 1124.73   33.04 1172.84      32 1194.97      32 1226.01   43.84 1235.14    45.4
 1261.36   51.84 1289.37   53.84 1388.34   53.84 1475.88   57.83 1549.58   55.84
 1929.04   55.84 2024.06   53.84 2101.65   61.84 2368.46   65.84 2519.88   71.84
 2528.36   73.84 3498.69   67.84 4057.72   67.84 4131.58   73.84 4486.93   79.74
#Mann= 3 ,-1 , 0
       0     .06       0  630.47    .035       0 2368.46     .06       0
Levee=0,,,-1,2598.81,73.87553,,	380
Bank Sta=1051.62,1235.14
XS Rating Curve= 0 ,0
Exp/Cntr=0.3,0.1

Type RM Length L Ch R = 1 ,36155.  ,323.19,333.66,348.72
XS GIS Cut Line= 5
 6414763.0731954 2043715.7192416 6414321.6532624 2044524.9890398
 6414132.4733249 2044819.2689794 6413838.1933854 2045491.9088412
 6412965.8635764   2047940.73835
#Sta/Elev= 30
       0   81.96  149.37   79.84  430.49   65.84  593.77   65.12  842.64   63.84
  911.84   55.84  945.72   47.84  953.66   49.33 1015.97   51.84 1043.98    39.5
 1184.61   30.99 1210.23   45.88 1224.79    54.1  1308.7    59.8 1369.41   56.42
 1679.83   55.84 1859.29   51.84  2063.4   67.26 2318.54   63.84 2369.36   65.84
 2409.21   73.84 2502.62   73.84 2534.49   65.84 2666.57   73.84 3310.38   73.08
 3349.24   72.76 3387.07   67.84 3793.69   67.84 4287.41   71.62 4605.43   79.19
#Mann= 3 ,-1 , 0
       0     .06       0  593.77    .035       0  2063.4     .06       0
Levee=0,,,-1,2670.33,75.14,,	380
Bank Sta=953.66,1210.23
XS Rating Curve= 0 ,0
Exp/Cntr=0.3,0.1

Type RM Length L Ch R = 1 ,35822.  ,862.61,848.98,790.43
XS GIS Cut Line= 5
 6414437.2632268 2043579.0892578 6414069.4133142 2044325.2990927
 6413827.6833757 2044661.6190236 6413470.3434728 2045365.7888671
 6412619.0336358 2047856.6583672
#Sta/Elev= 30
       0   81.84  157.88   79.84     323   73.84  431.11   65.84  616.74   64.72
  774.58   63.84  824.42   57.84  864.26   47.84  875.96   51.84  897.52   48.47
  941.69   48.02  988.21   43.84 1010.49    33.7 1130.63    30.9 1164.22   50.66
 1192.04   57.84 1298.37   57.84 1355.48   49.84 1587.98   49.84 1634.07   53.84
 1653.19   63.84 1666.69   65.84  1768.7   67.84 2181.32    64.7 2588.33   67.84
 2826.78   73.84 4339.45   71.84 4507.73   75.91 4568.38   79.84 4668.11   80.45
#Mann= 3 ,-1 , 0
       0     .06       0  616.74    .035       0  1768.7     .05       0
Levee=0,,,-1,2762.86,74.57,,	380
Bank Sta=897.52,1164.22
XS Rating Curve= 0 ,0
Exp/Cntr=0.3,0.1

Type RM Length L Ch R = 1 ,34973.  ,757.28,720.97,618.53
XS GIS Cut Line= 5
 6413638.5034382 2043035.1968962 6413362.6159919  2043810.309234
 6413139.2784994 2044230.7091476 6412823.9785878 2045465.6338643
 6412358.1305197 2047536.1201125
#Sta/Elev= 30
       0   81.25  589.19   77.84  604.08   73.84  649.58   71.84  662.62   65.84
   675.1   67.84  875.31    60.9     921   55.84  939.35   51.73  971.76   43.84
  981.99    33.7  1087.4    30.9 1098.45   37.84 1112.18   41.47 1174.44   43.84
 1219.33   43.84  1288.5   52.22 1365.81   57.84 1483.54   55.84 1717.92   59.84
 1740.77   51.84 1816.64   49.84 1883.64   51.84 1906.33   57.84 2046.95   59.84
 2153.04   65.84 2548.19   65.45 2803.38   73.84 4361.75   71.84 4695.57   75.83
#Mann= 3 ,-1 , 0
       0     .06       0  875.31    .035       0 2153.04     .06       0
Levee=0,,,-1,2796.42,74.19,,	380
Bank Sta=939.35,1174.44
XS Rating Curve= 0 ,0
Exp/Cntr=0.3,0.1

Type RM Length L Ch R = 1 ,34252.  ,678.44,652.64,592.59
XS GIS Cut Line= 6
  6412787.195968 2042663.4884821 6412627.4375539 2043633.4502685
 6412547.5583468 2043964.3783985 6412406.3630187 2045005.7454192
 6412270.9692171 2046061.8170245 6412056.8718027 2047399.1843019
#Sta/Elev= 30
       0   80.16     825   77.84  918.14   73.84     970   64.14 1001.12   51.77
  1032.6    37.5  1113.9   43.84 1156.11    33.7 1268.72    30.9 1316.59   51.12
 1347.24   55.84 1417.61   57.84 1437.97   51.84 1699.35   51.84 1723.34   53.84
  1738.2   48.84 1931.03   48.84 1958.92   57.84 2029.53   57.84  2040.8   53.84
 2092.51   57.84 2107.49   53.84 2126.81   53.84 2151.74   61.84 2223.73   61.84
 2231.78   63.84 2761.17   62.12 3204.93    73.8 4285.47   71.84 4793.47   77.57
#Mann= 3 ,-1 , 0
       0     .06       0     970    .035       0 2761.17     .05       0
Levee=0,,,-1,2852,72.5,,	380
Bank Sta=1001.12,1316.59
XS Rating Curve= 0 ,0
Exp/Cntr=0.3,0.1

Type RM Length L Ch R = 1 ,33599.  ,555.14,550.5,509.63
XS GIS Cut Line= 5
  6412273.686773 2042149.9792871 6411958.2476987 2043560.6967645
 6411931.9726745 2043928.5466771 6411945.1102102 2044729.9340391
 6411746.4840064   2047390.05527
#Sta/Elev= 30
       0   79.84 1444.77   77.84 1481.87   73.84  1497.6   63.84 1506.98    53.3
 1516.71    37.5 1531.67    34.2 1634.94    30.9 1644.72   37.84 1748.91   41.84
 1786.01   46.14 1828.86   57.84 1852.36   57.84 1859.64   53.84 1871.85   51.84
 2105.99   51.84 2112.11   53.84 2135.39   53.84 2147.47   48.84 2380.46   48.84
  2406.7   57.84 2549.17   57.84 2560.39   53.84  2575.8   53.84 2596.08   59.84
 2621.52   61.84 3188.61   63.84 3748.04   71.84 4909.13   71.84 5283.36   79.34
#Mann= 3 ,-1 , 0
       0     .06       0 1481.87    .035       0 2621.52     .06       0
Levee=0,,,-1,3232.02,72.5,,	380
Bank Sta=1506.98,1786.01
XS Rating Curve= 0 ,0
Exp/Cntr=0.3,0.1

Type RM Length L Ch R = 1 ,33049.  ,701.35,721.15,745.3
XS GIS Cut Line= 6
 6411878.0788058 2041852.8221331 6411510.2288458 2042772.4469383
 6411405.1288911 2043665.7967666 6411418.2663795 2043954.8217013
 6411470.8163806 2044716.7965034 6411381.3219238 2047481.3457788
#Sta/Elev= 30
       0   77.84  281.95   79.84 1082.55   74.05  1817.7   75.84 1882.94   73.84
 1896.07   63.84 1904.07   53.84 1920.95   49.21  1975.5    34.7 2101.17    30.9
 2144.39   49.42 2167.68   57.84 2206.58   57.84 2224.57   51.84 2443.89   51.84
 2456.81   53.84 2482.42   51.84 2657.89   51.84 2664.79   53.84 2864.66   51.84
 2904.43   53.84 2932.01   61.84 2943.09   61.84 3464.45   61.84    3613   65.84
 4194.16   71.84 5406.33   71.84 5648.91   77.84 5668.59   81.84 5709.08   81.84
#Mann= 3 ,-1 , 0
       0     .06       0 1882.94    .035       0 2943.09     .06       0
Levee=0,,,-1,3576.91,72,,	380
Bank Sta=1920.95,2144.39
XS Rating Curve= 0 ,0
Exp/Cntr=0.3,0.1

Type RM Length L Ch R = 6 ,33042.  ,,,
Node Name=South LS
Lateral Weir Pos= 0
Lateral Weir End=                ,                ,        ,Southside
Lateral Weir Distance=0
Lateral Weir TW Multiple XS=0
Lateral Weir WD=20
Lateral Weir Coef=2
Lateral Weir WSCriteria=-1
Lateral Weir Flap Gates= 0
Lateral Weir Hagers EQN= 0 ,,,,,
Lateral Weir SS=0.05,0.05,
Lateral Weir Type= 0
Lateral Weir Connection Pos and Dist= 0 ,
Lateral Weir SE= 27
       0   75.61  126.44   73.84  316.56   73.84  322.16   73.56  353.48   72.78
  395.98   71.84 1027.15   71.84 1041.47   71.16 1055.95   71.29 1105.99   71.34
 1311.88      70 2321.67      70 2361.29    68.1  2380.2   68.45  2385.2   68.94
 2459.27   69.06 2466.56   69.96 2892.25   69.95 3350.42   71.62 3440.53    71.6
 3468.49   70.35  3471.7   69.97 3473.22   69.94 3728.17   68.66 4117.38    68.1
 4895.43   69.26 5278.64   69.66
Lateral Weir HW RS Station=33049.  ,0
Lateral Weir TW RS Station=,0
LW Div RC= 0 ,False,

Type RM Length L Ch R = 1 ,32327.  ,622.82,600.26,528.79
XS GIS Cut Line= 5
 6410715.5872346  2043613.931172 6410674.3556182  2043963.853698
 6410715.4102991 2044743.8925881 6410879.6290227 2045955.0056514
 6410838.5743418 2047453.5014338
#Sta/Elev= 30
       0   70.38   21.98   65.76   25.61   63.84   35.66   53.84   48.49   51.67
  147.23    33.5  214.25    33.3  233.46    30.7  251.54      30  275.87   37.84
  281.86   43.84   296.1   45.84  313.23   51.26  341.05   57.84 1095.01   57.84
 1118.71   59.84 1182.55   61.84    1349   59.87 1531.27    60.3 1681.65   61.84
 1693.11   63.84 1773.32   65.84  2082.3   65.84 2122.68   67.84  2378.3   69.84
 2878.88   71.66 3428.02   71.84 3486.96   75.84 3593.66   79.84 3854.72   80.41
#Mann= 2 ,-1 , 0
       0    .035       0 1182.55     .06       0
Levee=0,,,-1,1752.85,70.00698,,	380
Bank Sta=48.49,313.23
XS Rating Curve= 0 ,0
Exp/Cntr=0.3,0.1

Type RM Length L Ch R = 1 ,31727.  ,761.92,772,797.79
XS GIS Cut Line= 4
 6410079.4474069 2043606.5299361 6410140.6447663 2044004.9083789
 6410284.5265989 2045466.3726105 6410284.3361731 2047453.5014338
#Sta/Elev= 30
       0   61.91    5.71   59.58   58.62    37.8   70.86    34.8  100.53   32.36
  140.15    32.8  167.32      30   175.1   37.84  203.94   45.84     268   45.06
  304.05   52.73  315.91   55.84  374.66   55.84  399.03   53.84  694.39   53.84
  713.58   55.84  729.16   55.84  736.66   53.84 1003.57   53.84 1032.07   57.84
 1050.96   57.84  1063.1   53.84 1105.93   51.84 1252.33   51.84 1309.18   57.84
 1379.44   59.84 2392.78   67.57 2932.65   69.84 3526.04   77.84 3858.71   79.84
#Mann= 2 ,-1 , 0
       0    .035       0 1379.44     .05       0
Levee=0,,,-1,1564.59,68.7301,,	380
Bank Sta=5.71,304.05
XS Rating Curve= 0 ,0
Exp/Cntr=0.3,0.1

Type RM Length L Ch R = 1 ,30955.  ,434.65,410.31,257.47
XS GIS Cut Line= 4
  6409322.941892 2043613.9722108 6409340.0785594 2044128.0724217
 6409565.8792808  2045236.548759  6409639.359792  2047542.883945
#Sta/Elev= 30
       0   66.13   21.18   56.38   58.08    37.8   78.76      32  126.07    32.3
  154.91    29.5  168.14   37.84  176.39   39.84  265.37   39.84  269.93   37.84
  284.83   37.84   356.1    55.4     389   55.84  405.97   53.84  804.13   53.84
  825.96   55.84   849.2   53.84    1290   53.84 1419.67   55.84 1431.34   57.84
    1461   55.84 1554.73   55.84 1878.57   61.65 2540.43   63.84 2951.43   67.84
 3137.14   69.84 3201.46   71.84 3208.22   73.84 3538.71   77.84 3953.13   77.99
#Mann= 2 ,-1 , 0
       0    .035       0 1419.67     .06       0
Levee=0,,,-1,1546.26,67.12914,,	380
Bank Sta=21.18,356.1
XS Rating Curve= 0 ,0
Exp/Cntr=0.3,0.1

Type RM Length L Ch R = 1 ,30545.  ,902.81,887.34,816.68
XS GIS Cut Line= 5
 6408902.9193746  2043613.931172 6408909.0044335 2043779.1076575
  6409052.695793  2044066.490424 6409360.6058762 2045318.6581209
 6409463.2426022 2047350.8647078
#Sta/Elev= 30
       0   69.98  154.46   69.84  178.25   63.84  192.02   56.49  196.98   53.84
  213.06   37.84  222.41    37.8  241.47   31.36  299.68    29.3  304.49   29.41
   341.4   41.84  415.07   43.84  462.86   55.45  486.59   55.84  527.81   55.84
  553.38   53.84  808.31   53.84  824.76   55.84  994.53   55.84 1003.71   53.84
  1357.1   53.84 1499.17   57.84 1512.08   53.84 1577.72   52.95  1817.5   59.38
  2791.9   63.84 3064.89   69.84 3197.12   69.84 3396.05   75.84 3810.86   77.84
#Mann= 2 ,-1 , 0
       0    .035       0  486.59     .05       0
Levee=0,,,-1,1613.59,66.62889,,	380
Bank Sta=192.02,462.86
XS Rating Curve= 0 ,0
Exp/Cntr=0.3,0.1

Type RM Length L Ch R = 1 ,29658.  ,857.08,844.81,775.99
XS GIS Cut Line= 5
 6408009.7468605 2043692.6432103 6408087.9108625 2044148.5997858
 6408272.6569029  2044456.509869 6408560.0396694 2045113.3847163
 6409032.1684762 2047474.0287506
#Sta/Elev= 30
       0   71.55  456.95   69.84  503.24   67.47  545.73    56.4  555.68   51.78
  563.54   43.84  584.14   37.84  636.55   38.01  684.92    29.5  750.91      29
  761.66   37.84  799.77   49.98  824.81   57.84  943.13   60.39 1131.47   59.95
  1289.3   53.84 1705.87   53.84 1729.09   57.84 1745.78   57.84 1761.82   55.84
 1862.84   55.23 2090.23   57.84 2244.32   61.84 2463.75   63.84 2899.89   63.84
  2916.6   65.84 3243.16   67.84 3350.31   71.84  3360.7   73.84 3946.07   77.63
#Mann= 2 ,-1 , 0
       0    .035       0 1745.78     .05       0
Levee=0,,,-1,1860.77,65.0979,,	380
Bank Sta=555.68,799.77
XS Rating Curve= 0 ,0
Exp/Cntr=0.3,0.1

Type RM Length L Ch R = 1 ,28813.  ,668.58,698.93,673.99
XS GIS Cut Line= 5
 6407039.1905082 2043728.8185786 6407400.1680035 2044669.5066666
 6407658.4019393 2045008.4386926 6407932.7754932 2045508.7669463
 6408578.3603092 2047574.6383858
#Sta/Elev= 30
       0    68.4  986.21   67.64 1006.19   65.79 1062.14   53.84 1077.04   47.91
 1090.21   37.84 1097.92   37.57 1131.31    37.5 1148.43   31.34  1167.2    29.5
 1237.24    28.4 1243.06   37.84 1323.58   43.84 1334.11   48.68 1379.66   65.84
 1819.57   61.84 1869.55   53.84 1925.69   51.84 1957.69   53.84 2007.52   64.56
 2154.01   62.91 2285.24   55.84 2364.68   55.84  2484.5   61.84 2636.54   63.84
 3219.63   63.84 3511.44   67.84 3583.49   71.84 3776.76   76.41 4168.68   78.13
#Mann= 3 ,-1 , 0
       0     .06       0 1006.19    .035       0 2154.01     .06       0
Levee=0,,,-1,2569.44,69.04,,	380
Bank Sta=1097.92,1334.11
XS Rating Curve= 0 ,0
Exp/Cntr=0.3,0.1

Type RM Length L Ch R = 1 ,28114.  ,360.35,390.56,451.68
XS GIS Cut Line= 6
 6406383.6799769 2043692.2465963 6406803.0020416 2044782.4839928
 6406883.7001317 2045137.5556842 6407319.4699133 2045718.5819807
 6407665.1485421 2046418.4992649 6408216.2795937 2047433.7407431
#Sta/Elev= 30
       0   69.36  1135.8      65 1532.22   53.91 1538.58   53.84 1558.21    44.4
 1571.87   39.84 1609.75      37 1646.74      37 1662.86    31.5 1673.88   32.42
 1678.95      30 1756.66    28.4 1778.32   39.84 1798.21   47.61 1815.18   53.84
 1823.77   55.84 1843.18   59.84 2044.01   61.84 2059.64   63.84 2539.62   63.59
 2784.66    60.9  3268.8   61.84 3358.53   64.14 3393.88   67.84 3462.99   69.84
 3740.63   69.84 3770.26   71.84 3853.73   73.06 4039.32      74 4194.32   75.78
#Mann= 3 ,-1 , 0
       0     .06       0 1532.22    .035       0 1823.77     .05       0
Levee=0,,,-1,4002.5,73.93548,,	380
Bank Sta=1558.21,1798.21
XS Rating Curve= 0 ,0
Exp/Cntr=0.3,0.1

Type RM Length L Ch R = 1 ,27723.  ,624.48,685.03,705.83
XS GIS Cut Line= 5
 6405892.9099351 2043073.4349505  6406566.613635 2045308.1594714
 6406730.9316186  2045653.227204 6407263.6861287 2046656.2023339
 6407520.7882071 2047588.1972914
#Sta/Elev= 30
       0      75  104.87    74.7  415.72      70 1659.09      65 1763.01   63.03
 1933.44    62.2 2334.07   54.68 2387.62   53.84 2396.83   49.29 2407.87   43.84
 2420.33   39.84 2444.04   38.88  2469.9   35.07 2490.44      34 2500.08    31.2
 2595.07    28.5 2605.65   39.84 2654.85   54.53 2685.28   57.84 2724.49   59.84
 2734.86   61.84 2764.91   63.84 3143.26   63.84 3265.17   61.84 3362.84   57.84
 3428.83   57.84 3557.37   60.74 3675.82   65.84 3900.81   69.84 4818.76   70.47
#Mann= 3 ,-1 , 0
       0     .06       0 2334.07    .035       0 2734.86     .06       0
Bank Sta=2396.83,2654.85
XS Rating Curve= 0 ,0
Exp/Cntr=0.3,0.1

Type RM Length L Ch R = 6 ,27470.  ,,,
Node Name=North LS
Lateral Weir Pos= 3
Lateral Weir End=                ,                ,        ,Northside
Lateral Weir Distance=0
Lateral Weir TW Multiple XS=0
Lateral Weir WD=20
Lateral Weir Coef=2
Lateral Weir WSCriteria=-1
Lateral Weir Flap Gates= 0
Lateral Weir Hagers EQN= 0 ,,,,,
Lateral Weir SS=0.05,0.05,
Lateral Weir Type= 0
Lateral Weir Connection Pos and Dist= 0 ,
Lateral Weir SE= 30
       0   69.84   248.5   67.84 2091.82   67.81 2313.68   65.84 2609.55   65.84
 2635.68   67.84 2831.04   67.84 3021.44   65.89 3066.15   65.84 3242.95   66.84
 3316.39   67.84 3476.85   67.28  3786.3   68.92 3830.66   69.84 3949.75   69.84
 3962.76   65.84 4126.04   63.84 4267.12   64.43 4300.91   65.45 4371.78   65.47
 4461.03   64.84 4626.77   64.81 4670.04   65.14 4689.74   64.55    4804   64.17
  5054.3   64.79 5130.79   65.84 5467.54   66.53 5499.43   66.38 5512.54   65.28
LW Div RC= 0 ,False,

Type RM Length L Ch R = 1 ,27038.  ,481.08,641.78,711.72
XS GIS Cut Line= 5
 6405580.7057804  2043155.593966 6405818.4851523 2044750.2047568
 6405979.8813799 2045637.8838906 6406141.2776076  2046025.234818
 6406243.6811175 2046864.6507802
#Sta/Elev= 30
       0      75  457.66   69.59 1384.39      65 1648.72      60 2398.35      60
 2553.29   53.84 2573.53   46.64 2589.69   39.84 2625.55      39 2666.92   32.53
 2675.15      33 2683.12    30.9 2690.27    31.3 2700.57   39.84 2743.13   39.84
 2746.91   35.24 2749.25   30.66 2764.97      32 2780.18    29.5 2801.52      29
 2816.67   39.84 2844.85   49.84 2859.58   51.84 2869.79   51.84 3112.11   47.84
 3199.21   49.84 3307.93   59.84 3407.34   64.46 3560.66   67.84 3779.74   67.84
#Mann= 3 ,-1 , 0
       0     .06       0 2553.29    .035       0 2869.79     .06       0
Bank Sta=2573.53,2859.58
XS Rating Curve= 0 ,0
Exp/Cntr=0.3,0.1

Type RM Length L Ch R = 1 ,26396.  ,407.87,468.66,469.88
XS GIS Cut Line= 5
 6405501.4660595 2043204.3421721 6405463.4135082 2044685.6462847
 6405447.2738902 2045654.0235086 6405463.4135082  2046331.887608
 6405478.1409552 2046655.8671125
#Sta/Elev= 30
       0    74.5   479.1    67.5 1009.06      65 1126.68      60 2324.36      60
    2440   49.75 2506.02      45 2586.93   44.52 2611.51   43.76 2665.22   41.84
 2735.19   41.62 2762.94   39.84 2771.45   35.91 2779.85    34.6 2787.26      32
 2802.36    30.7 2853.41    31.5 2861.18   29.99 2883.69    29.5 2923.54   39.84
 2931.39   43.84 2945.98   47.84 2969.72   48.26 3060.94   49.84  3090.4   51.84
 3096.23   53.84  3123.8   57.84 3146.39   63.84 3159.68   65.84 3452.68   68.04
#Mann= 3 ,-1 , 0
       0     .06       0 2586.93    .035       0 2969.72     .06       0
Bank Sta=2611.51,2969.72
XS Rating Curve= 0 ,0
Exp/Cntr=0.3,0.1

Type RM Length L Ch R = 1 ,25928.  ,309.94,393.16,426.71
XS GIS Cut Line= 5
    6405366.5758  2043200.801189 6405092.2022461 2045153.6953023
 6404979.2249199 2045750.8612641 6404995.3645379 2046283.4687066
 6404970.1599786 2046590.9640941
#Sta/Elev= 30
       0   74.48     565      65  775.98   63.66   951.6      65 1013.53      60
 1814.98      60 2370.61      65 2435.44   62.36 2483.98   62.15 2605.76   52.63
 2688.69   43.84 2761.89   43.84 2776.31   39.84 2825.38    34.6 2839.11    34.6
  2847.3    31.5 2899.18    30.9 2912.97      32 2920.64      30 2940.12    29.5
 2967.36   39.84 2974.86   43.84 2988.52   47.84 3007.99    50.4 3053.41   51.98
  3067.8   53.84 3111.33   65.84 3137.12   67.84 3263.63   67.84 3421.21   65.84
#Mann= 2 ,-1 , 0
       0     .06       0 2605.76    .035       0
Bank Sta=2605.76,3007.99
XS Rating Curve= 0 ,0
Exp/Cntr=0.3,0.1
